--- WILLIAMSRV.prj (project) ---

Proj Title=WILLIAMSRV
Current Plan=p01
Default Exp/Contr=0,0
English Units
Geom File=g01
Flow File=f01
Plan File=p01
Background Map Layer=Inundation Boundary (01pct Value_0)
BEGIN DESCRIPTION:
----------MODEL BY WOOD PLC 2021----------
Stream Name: Williams River
Flood Zone: Approximate
Pocahontas County, WV
HEC-RAS Version: RAS 6.1
Vertical Datum: NAVD88
Projection: NAD 1983 StatePlane West Virginia S FIPS 4702 (US Feet)
Terrain: 1-meter LIDAR (FEMA Region III 3DEP collected 2016-2018)
Land Use: 2019 NLCD
Hydrologic Method:
WV 2010 Regional Regression Equations
Model Notes:
Model extends county boundary at the downstream
END DESCRIPTION:
DSS Export Rating Curves= 0
DSS Export Rating Curve Sorted= 0
DSS Export Volume Flow Curves= 0
DXF Filename=..\CHARLESCK\CHARLESCK.
DXF OffsetX= 0
DXF OffsetY= 0
DXF ScaleX= 0
DXF ScaleY= 0

--- WILLIAMSRV.p01 (plan) ---

Plan Title=Floodplain
Program Version=6.00
Short Identifier=Floodplain
Geom File=g01
Flow File=f01
Subcritical Flow
K Sum by GR= 0
Std Step Tol= 0.01
Critical Tol= 0.01
Num of Std Step Trials= 20
Max Error Tol= 0.3
Flow Tol Ratio= 0.001
Split Flow NTrial= 30
Split Flow Tol= 0.02
Split Flow Ratio= 0.02
Log Output Level= 0
Friction Slope Method= 1
Unsteady Friction Slope Method= 2
Unsteady Bridges Friction Slope Method= 1
Parabolic Critical Depth
Global Vel Dist= 0 , 0 , 0
Global Log Level= 0
CheckData=True
Encroach Param=-1 ,0,0, 0
Mapping Interval=1HOUR
Computation Time Step Use Courant=        0
Computation Time Step Use Time Series=    0
Computation Time Step Count To Double=0
Computation Time Step Max Doubling=0
Computation Time Step Max Halving=0
Computation Time Step Residence Courant=0
Run HTab= 0
Run UNet= 0
Run Sediment= 0
Run PostProcess= 0
Run WQNet= 0
Run RASMapper=-1
UNET Theta= 0
UNET Theta Warmup= 0
UNET ZTol= 0
UNET ZSATol= 0
UNET MxIter= 0
UNET Max Iter WO Improvement= 0
UNET MaxInSteps= 0
UNET DtIC= 0
UNET DtMin= 0
UNET MaxCRTS= 0
UNET WFStab= 0
UNET SFStab= 0
UNET WFX= 1
UNET SFX= 1
UNET Gravity=32.174
UNET 1D Methodology=Finite Difference
UNET DSS MLevel= 1
UNET Pardiso=0
UNET DZMax Abort= 0
UNET Use Existing IB Tables= 0
UNET Froude Reduction=False
UNET Froude Limit= 0
UNET Froude Power= 0
UNET D1 Cores= 0
UNET WindReference=Eulerian
UNET WindDragFormulation=Hsu (1988)
UNET D2 Coriolis=0
UNET D2 Cores= 0
UNET D2 Theta= 1
UNET D2 Theta Warmup= 1
UNET D2 Z Tol= 0.01
UNET D2 Volume Tol= 0.01
UNET D2 Max Iterations= 20
UNET D2 Equation= 0
UNET D2 RampUpFraction=0.1
UNET D2 TimeSlices= 1
UNET D2 Turbulence Formulation=Non-Conservative (original)
UNET D2 Eddy Viscosity=0.3
UNET D2 Transverse Eddy Viscosity=0.1
UNET D2 Smagorinsky Mixing=0
UNET D2 BCVolumeCheck=0
UNET D2 Cores=0
UNET D2 SolverType=PARDISO (Direct)
UNET D2 Minimum Iterations= 2147483647
UNET D2 Maximum Iterations= 2147483647
UNET D2 Restart Number= 10
UNET D2 Relaxation Coeff=1.3
UNET D2 SOR Precondition Iterations= 10
UNET D2 ILUT Maximum Fill= 8
UNET D2 ILUT Tolerance=1E-08
UNET D1D2 MaxIter= 0
UNET D1D2 ZTol=0.01
UNET D1D2 QTol=0.1
UNET D1D2 MinQTol=1
Write IC File= 0
Write IC File at Fixed DateTime=0
Write IC File at Sim End=0
Echo Input=False
Echo Parameters=False
Echo Output=False
Write Detailed= 0
HDF Write Warmup=0
HDF Write Time Slices=0
HDF Flush=0
HDF Compression= 1
HDF Chunk Size= 1
HDF Spatial Parts= 1
HDF Use Max Rows=0
HDF Fixed Rows= 1
Calibration Method= 0
Calibration Iterations= 20
Calibration Max Change=0.05
Calibration Tolerance=0.2
Calibration Maximum=1.5
Calibration Minimum=0.5
Calibration Optimization Method= 1
WQ AD Non Conservative
WQ ULTIMATE=-1
WQ Max Comp Step=1HOUR
WQ Output Interval=15MIN
WQ Output Selected Increments= 0
WQ Output face flow=0
WQ Output face velocity=0
WQ Output face area=0
WQ Output face dispersion=0
WQ Output cell volume=0
WQ Output cell surface area=0
WQ Output cell continuity=0
WQ Output cumulative cell continuity=0
WQ Output face conc=0
WQ Output face dconc_dx=0
WQ Output face courant=0
WQ Output face peclet=0
WQ Output face adv mass=0
WQ Output face disp mass=0
WQ Output cell mass=0
WQ Output cell source sink temp=0
WQ Output nsm pathways=0
WQ Output nsm derived pathways=0
WQ Create Restart=0
WQ Fixed Restart=0
WQ System Summary=0
WQ Write To DSS=0
Sorting and Armoring Iterations= 10
XS Update Threshold= 0.02
Bed Roughness Predictor= 0
Hydraulics Update Threshold= 0.02
Energy Slope Method= 1
Volume Change Method= 1
Sediment Retention Method= 0
Sediment TS Multiplier= 1
Warm Up Method= 0
XS Weighting Method= 0
Number of US Weighted Cross Sections= 1
Number of DS Weighted Cross Sections= 1
Upstream XS Weight=0
Main XS Weight=1
Downstream XS Weight=0
Number of DS XS's Weighted with US Boundary= 1
Upstream Boundary Weight= 1
Weight of XSs Associated with US Boundary= 0
Number of US XS's Weighted with DS Boundary= 1
Downstream Boundary Weight= 0.5
Weight of XSs Associated with DS Boundary= 0.5
Percentile Method= 0
Sediment Output Level= 3
Mass or Volume Output= 0
Output Increment Type= 1
Profile and TS Output Increment= 1
Transport Output Increment 1
XS Output Flag= 0
XS Output Increment= 10
Read HDF5 Sediment Hotstart= 0
Sediment Hotstart Type= 0
Write Gradation File= 0
Read Gradation Hotstart= 0
Write HDF5 File= 1
Write Binary Output= 1
Write DSS Sediment File= 0
DSS Sediment Output Type= 1
SV Curve= 0
Specific Gage Flag= 0
Subcell Erosion Methods= 0
Subcell Deposition Methods= 0
Advection Scheme= 1
Matrix Solver= 0
Implicit Weighting Factor= 1
Maximum Outer Loop Convergence Iterations= 5
Convergence Maximum Absolute= 0.001
Convergence RMSE= 0.0001
Grain Fractions Max Abs Error= 0.001
Max Subgrid Regions= 1
Max Subgrid Length Scale= 3.402823E+38
Initial Layer Thickness= 3.402823E+38
Min Layer Thickness= 3.402823E+38
Max Layer Thickness= 3.402823E+38
Number of Layers= 5

--- WILLIAMSRV.f01 (steady flow) ---

Flow Title=Flow
Program Version=6.00
Number of Profiles= 6
Profile Names=01pct,10pct,04pct,02pct,0_2pct,01plus
River Rch & RM=WILLIAMSRV,Main            ,87980
     575     304     404     487     803     850
River Rch & RM=WILLIAMSRV,Main            ,82791
     969     523     688     824    1340    1430
River Rch & RM=WILLIAMSRV,Main            ,77773
    1370     747     977    1170    1880    2020
River Rch & RM=WILLIAMSRV,Main            ,76516
    1530     837    1090    1300    2090    2260
River Rch & RM=WILLIAMSRV,Main            ,70859
    1810     998    1300    1540    2470    2670
River Rch & RM=WILLIAMSRV,Main            ,63528
    2110    1170    1520    1800    2870    3120
River Rch & RM=WILLIAMSRV,Main            ,62377
    2410    1350    1740    2060    3270    3560
River Rch & RM=WILLIAMSRV,Main            ,53448
    2730    1530    1980    2340    3700    4040
River Rch & RM=WILLIAMSRV,Main            ,45382
    3450    1950    2510    2960    4650    5100
River Rch & RM=WILLIAMSRV,Main            ,34732
    4490    2570    3290    3870    6030    6640
River Rch & RM=WILLIAMSRV,Main            ,34489
    5120    2950    3760    4420    6870    7580
River Rch & RM=WILLIAMSRV,Main            ,28469
    5700    3290    4190    4920    7620    8430
River Rch & RM=WILLIAMSRV,Main            ,20081
    7070    4120    5220    6120    9420   10500
River Rch & RM=WILLIAMSRV,Main            ,14524
    8070    4720    5980    6990   10700   11900
Boundary for River Rch & Prof#=WILLIAMSRV,Main            , 1
Up Type= 0
Dn Type= 3
Dn Slope=0.01
Boundary for River Rch & Prof#=WILLIAMSRV,Main            , 2
Up Type= 0
Dn Type= 3
Dn Slope=0.01
Boundary for River Rch & Prof#=WILLIAMSRV,Main            , 3
Up Type= 0
Dn Type= 3
Dn Slope=0.01
Boundary for River Rch & Prof#=WILLIAMSRV,Main            , 4
Up Type= 0
Dn Type= 3
Dn Slope=0.01
Boundary for River Rch & Prof#=WILLIAMSRV,Main            , 5
Up Type= 0
Dn Type= 3
Dn Slope=0.01
Boundary for River Rch & Prof#=WILLIAMSRV,Main            , 6
Up Type= 0
Dn Type= 3
Dn Slope=0.01
DSS Import GetInterval= 0
DSS Import GetPeak= 0
DSS Import FillOption= 0

--- WILLIAMSRV.g01 (geometry) ---

Geom Title=Geometry
Program Version=6.10

River Reach=WILLIAMSRV      ,Main
Reach XY= 30
2203807.40824081451136.6289569742204002.18534918  449482.5029463
2202725.89939801448526.1065300262199813.50612365449162.107971638
2196740.21448199451892.4403274662196972.61906929453381.596569076
2193385.91587083456876.1052581072190893.45059304456401.774239585
2189746.30480142457972.2022280542190692.70776422462519.158357233
2192493.05619763465162.2327954922192725.78866467468253.013194654
2194890.38904328471677.2158178892196911.23708554473369.319645658
2197696.45417829477973.4122048912197023.13965715480225.178063229
2196379.49704222481316.6398802252195771.19735293481016.382145479
2194249.51397081484324.3316103222191883.46161635 485275.42485249
2191053.66635992486821.6117207412189439.04050104486678.102292836
2187385.90433849491577.0982727262184778.67103593 493090.67661041
 2181367.0751688492838.4048052432180391.20474525494764.456399322
2178568.72348209495863.8597123322178834.92472129497116.534700409
2177145.91956915498537.6745746432176627.81168149500275.048724562

Type RM Length L Ch R = 1 ,87980   ,351.6,375.9,359.7
XS GIS Cut Line= 4
2204129.68369501 451217.054249162203876.02572586451142.854979274
2203625.81888555451056.5767584772203332.47293484450946.140635856
#Sta/Elev= 30
       0 3486.37      43 3483.14    80.8 3481.23   113.5 3478.35   147.4 3476.87
   193.3 3473.46   222.5  3472.2   255.8 3472.28   264.1 3471.61   276.8 3472.43
   302.2 3470.53   314.9 3471.09   323.4 3470.51   331.6 3469.69   340.3 3470.49
   355.3 3470.54   371.1 3471.51   429.1 3470.81   453.5 3471.73   473.1 3474.63
     492 3475.72   616.7 3478.31   693.1  3483.9   710.2 3484.28   718.8 3485.65
   747.1 3487.83   757.2 3489.63   791.4 3492.28   821.3 3495.59842.3976  3496.7
#Mann= 6 ,-1,0
       0      .1       0   323.4    .045       0   340.3      .1       0
  364.29     .12       0  678.95      .1       0  698.95     .12       0
Bank Sta=323.4,340.3
XS Rating Curve= 0 ,0
Exp/Cntr(USF)=0,0
Exp/Cntr=0.3,0.1

Type RM Length L Ch R = 1 ,87604   ,287.3,278.9,229.2
XS GIS Cut Line= 4
2204190.07844957 451008.260954832204012.34531472450932.336120529
 2203825.9843578 450808.095482582203473.96921695450657.971378392
#Sta/Elev= 30
       0 3486.45    67.3 3480.79    89.1 3479.49   119.6 3474.06   180.4 3471.85
   231.9    3471   247.6  3468.2     256 3466.75     269 3468.22   275.2 3468.54
   285.5 3468.09   294.4 3469.44   319.7 3468.81   350.4 3469.73   409.8 3469.95
   427.9 3471.86     441 3475.35   445.3 3475.75   467.1 3475.54   484.9 3473.74
   527.9 3474.33   567.4 3475.82   646.4 3477.67   695.2 3480.34   710.2  3480.2
   722.7 3482.53   749.7 3489.16   753.1 3488.94   784.5 3491.98799.9393 3495.72
#Mann= 7 ,-1,0
       0     .12       0      30      .1       0   247.6    .045       0
     269     .12       0  467.25      .1       0  567.25     .12       0
  687.25      .1       0
Bank Sta=247.6,269
XS Rating Curve= 0 ,0
Exp/Cntr(USF)=0,0
Exp/Cntr=0.3,0.1

Type RM Length L Ch R = 1 ,87325   ,460.2,463.7,450.6
XS GIS Cut Line= 4
2204278.08223478450747.7007280222204145.21377475450721.817261783
2203893.28137002450687.3059734642203510.20606968450533.730740444
#Sta/Elev= 30
       0 3492.72    34.5 3487.32    71.2 3480.11    87.5 3479.18    95.7 3477.08
   103.8 3476.49     130 3471.54   152.6 3470.26   164.7 3468.22   176.8 3468.18
  184.043467.065   188.9 3466.52  227.173467.064   233.3 3467.82   257.6 3467.41
     286 3468.71   318.1  3467.8   362.5 3469.92   395.2 3476.53   412.4 3475.77
   490.6 3475.69   520.1 3474.18   567.4 3476.33   599.6 3475.24     658 3477.67
   699.8 3482.03   735.6 3487.83   748.5 3488.15   761.5 3489.68802.3643 3500.97
#Mann= 3 ,-1,0
       0     .12       0  184.04    .045       0  227.17     .12       0
Bank Sta=184.04,227.17
XS Rating Curve= 0 ,0
Exp/Cntr(USF)=0,0
Exp/Cntr=0.3,0.1

Type RM Length L Ch R = 1 ,86861   ,486,487.2,481.7
XS GIS Cut Line= 4
2204459.26649846450340.4675258582204224.58973789450355.997605601
2203977.83402641450328.3885749462203596.48429048450259.365998308
#Sta/Elev= 30
       0 3488.36    43.2 3486.09    56.2  3484.5    99.3 3482.41   171.5 3474.51
   202.9 3473.66   267.8 3470.08   287.9  3468.2   299.7 3464.59   308.1 3462.76
   312.1 3463.02   317.8 3464.46   328.2 3464.72   339.5 3465.88   372.5 3464.96
   384.5 3465.77   416.7 3465.82   424.8 3468.29   432.8 3472.18   436.4    3473
     461 3474.55     538 3475.98   607.1 3474.74   668.1    3476   680.3 3477.58
   765.7 3483.56     786 3486.94     794 3487.03   830.7 3490.48871.0313 3496.88
#Mann= 6 ,-1,0
       0     .12       0     180      .1       0   299.7    .045       0
   317.8      .1       0  385.19     .12       0  603.49      .1       0
Bank Sta=299.7,317.8
XS Rating Curve= 0 ,0
Exp/Cntr(USF)=0,0
Exp/Cntr=0.3,0.1

Type RM Length L Ch R = 1 ,86374   ,396.1,393.9,388
XS GIS Cut Line= 4
2204511.03343093450107.5163297042204241.84538205450069.553912553
2203972.65733316450088.535121129 2203620.6421923450073.005041385
#Sta/Elev= 30
       0  3486.8    54.2 3483.53    95.8 3482.83   148.3 3479.29   192.7 3470.14
   237.2 3468.01   281.5 3467.64   289.6 3466.76  302.883462.631   309.6 3461.58
  315.953462.633   321.6 3463.62   365.8 3464.35   393.8 3464.44   405.9 3463.31
   421.9 3464.67     446 3465.25   471.6 3468.03   485.5 3468.36   518.1 3472.28
   566.2 3474.24   614.1 3473.93   658.3 3471.43   810.5 3475.73   822.5 3479.15
   842.5 3486.32   854.5 3488.01   866.5 3491.77   886.4 3495.26894.0657 3497.42
#Mann= 4 ,-1,0
       0     .12       0     140      .1       0  302.88    .045       0
  315.95      .1       0
Bank Sta=302.88,315.95
XS Rating Curve= 0 ,0
Exp/Cntr(USF)=0,0
Exp/Cntr=0.3,0.1

Type RM Length L Ch R = 1 ,85980   ,251.6,258.9,253.3
XS GIS Cut Line= 4
2204252.19876854449729.6177226112204083.09345578449777.933526258
2203900.18362769449843.5049740642203636.17227205449826.249329904
#Sta/Elev= 30
       0 3484.04    20.8  3483.2    74.9 3478.56    90.3 3473.26   112.3 3461.85
   116.5 3460.62   153.9 3462.38   164.7 3461.18     179 3461.73   191.7 3460.65
     230 3460.67     247 3461.57   265.1 3461.05   272.5 3459.79   276.7 3460.05
   280.3 3461.28   285.2 3461.94   336.2  3462.1   344.7 3464.03   361.7 3471.68
   365.9 3472.71   386.2 3473.43   398.2 3474.86   470.4 3472.74   494.5 3473.65
     535 3479.96   578.6  3490.3   598.7 3494.21   618.7 3501.74634.7549 3504.62
#Mann= 4 ,-1,0
       0     .12       0  175.87      .1       0   265.1    .045       0
   280.3      .1       0
Bank Sta=265.1,280.3
XS Rating Curve= 0 ,0
Exp/Cntr(USF)=0,0
Exp/Cntr=0.3,0.1

Type RM Length L Ch R = 1 ,85721   ,236.6,234.3,230.3
XS GIS Cut Line= 4
2204209.05965814449553.6101521842204038.22878096449626.083857654
2203870.84903262449686.4786122122203639.62340088449722.715464947
#Sta/Elev= 30
       0 3487.45    18.3 3484.59      27 3484.02    48.8 3480.43    61.8 3479.34
    88.8 3471.66    96.6 3470.23   118.3 3469.22     153 3465.68     209 3463.74
   238.8 3461.13   281.3 3460.67   289.8 3458.93   298.3 3459.52   300.8  3460.7
   306.8 3462.88   336.5 3464.32   359.7 3467.05   422.9 3467.93   451.2 3467.64
   463.4 3468.29   479.6  3473.7   487.7 3475.83   501.2 3481.53     516 3486.06
   529.2 3489.19   548.4 3495.97   564.6 3499.19   588.9  3503.1597.5587 3503.87
#Mann= 3 ,-1,0
       0      .1       0   281.3    .045       0   300.8      .1       0
Bank Sta=281.3,300.8
XS Rating Curve= 0 ,0
Exp/Cntr(USF)=0,0
Exp/Cntr=0.3,0.1

Type RM Length L Ch R = 1 ,85487   ,294.5,297.1,286.6
XS GIS Cut Line= 4
2204062.27285655 449410.547166082204013.41458927449444.928909722
2203805.31456196449602.3611042922203656.93019466449687.410680669
#Sta/Elev= 30
       0 3483.96    12.3 3483.58    14.9 3482.84    51.5 3469.11    80.8 3459.58
    89.4 3458.55    95.1 3459.58    99.9 3460.17   126.5 3460.22   146.3 3459.91
   156.6 3458.78   172.9 3461.01   191.7 3460.74     215 3462.53   232.1    3462
   257.8 3463.43     292 3463.28   307.1 3462.42   326.5 3463.99   344.1 3464.36
   363.5 3463.17   379.3  3463.8   386.5 3465.35   400.4 3470.48   430.9 3486.17
   437.3  3488.5   455.7 3493.15   464.9 3494.07   478.9 3497.88   491.7  3499.2
#Mann= 4 ,-1,0
       0     .12       0      30      .1       0    80.8    .045       0
    95.1      .1       0
#XS Ineff= 2 , 0
                          216.45         3464.32
Permanent Ineff=
       F       F
Bank Sta=80.8,95.1
XS Rating Curve= 0 ,0
Exp/Cntr(USF)=0,0
Exp/Cntr=0.3,0.1

Type RM Length L Ch R = 1 ,85190   ,469.7,479,468.5
XS GIS Cut Line= 4
2203951.95056017449293.0499253762203898.45806327449344.816857854
2203682.76251128449570.865796344 2203630.9955788449641.613937398
#Sta/Elev= 30
       0 3487.72     8.4 3486.35    23.2 3484.91    45.2 3481.38    57.7 3478.02
    63.5 3474.57    72.1 3467.34    79.1 3460.71   81.36  3459.3    84.8  3458.4
    97.1 3458.23  104.78 3459.22   124.4 3460.61   153.1  3459.2   168.9 3460.95
     182 3461.23     198 3460.56     263 3459.97     280 3459.21   353.6 3459.18
     379 3460.38   384.6 3461.98   401.8  3473.9   409.6 3477.76   419.5 3483.38
   425.1 3485.87   444.8 3490.74   452.2 3491.39   464.1 3494.24474.5508 3495.74
#Mann= 4 ,-1,0
       0     .12       0   81.36    .045       0  104.78     .12       0
  184.44      .1       0
#XS Ineff= 2 , 0
                          309.58         3463.94
Permanent Ineff=
       F       F
Bank Sta=81.36,104.78
XS Rating Curve= 0 ,0
Exp/Cntr(USF)=0,0
Exp/Cntr=0.3,0.1

Type RM Length L Ch R = 1 ,84711   ,362.9,370.7,361.1
XS GIS Cut Line= 4
2203725.90162168449236.1062996492203605.11211256449331.012342527
2203439.45792863449460.4296737232203356.63083666449544.982330104
#Sta/Elev= 30
       0 3480.04    12.4 3477.96    32.7 3476.65    40.6 3475.62    53.5 3472.62
    68.3 3470.51    79.4 3466.65    98.8 3462.47   124.3 3460.66   139.5 3458.56
   172.9 3457.07   185.3  3457.4   198.6 3456.89   241.6 3457.96   276.6  3457.2
  282.95  3456.4   291.9 3455.17     302 3456.47   327.4 3456.06   332.5 3457.88
   345.6 3460.39   357.8 3463.85   374.2 3472.23   397.1 3475.05   406.3 3477.67
   415.3 3478.66   437.1  3482.9   454.5 3484.16   471.3 3487.07482.1902 3487.85
#Mann= 6 ,-1,0
       0     .12       0      50      .1       0     150     .12       0
  173.61      .1       0  282.95    .045       0     302      .1       0
Bank Sta=282.95,302
XS Rating Curve= 0 ,0
Exp/Cntr(USF)=0,0
Exp/Cntr=0.3,0.1

Type RM Length L Ch R = 1 ,84340   ,184.8,269.1,275.7
BEGIN DESCRIPTION:
structure xs 4
END DESCRIPTION:
XS GIS Cut Line= 4
2203572.32638866449079.079937798 2203511.9316341449118.767919365
2203348.00301458449244.7341217292203237.56689196449322.384520447
#Sta/Elev= 30
       0 3481.07    33.7 3478.72    40.2    3478    47.5 3476.44    59.4 3472.67
      77 3462.56    88.1 3457.52    92.1 3456.15   110.9  3455.4   122.4 3455.68
   127.5 3455.17  129.32 3454.54   135.3 3453.36  146.07 3454.54   153.7 3455.74
   181.3 3455.73     205  3456.5   233.4 3456.24   248.5 3457.33   263.7  3457.5
   268.7 3459.14   293.7 3471.96     305 3473.83   317.9 3474.95   327.7 3476.39
   333.8 3476.59   342.4 3477.88   352.1 3478.12     391 3483.16414.0074 3484.84
#Mann= 3 ,-1,0
       0      .1       0  129.32    .045       0  146.07      .1       0
Bank Sta=129.32,146.07
XS Rating Curve= 0 ,0
Exp/Cntr(USF)=0,0
Exp/Cntr=0.5,0.3

Type RM Length L Ch R = 1 ,84071   ,125.5,48.3,48.5
BEGIN DESCRIPTION:
structure xs 3
END DESCRIPTION:
XS GIS Cut Line= 5
2203488.42856772448956.8147519992203356.58694276 449018.77626935
2203295.79298181449022.0485026132203203.31443831  449068.8818521
2203062.14601344449162.528232953
#Sta/Elev= 30
       0 3482.57    10.3 3481.72    40.1 3477.74    44.5 3476.26    57.7 3468.42
    69.6 3463.37    75.4 3462.15    93.1    3460   104.3 3459.28   117.7 3457.76
   132.5 3457.45   148.4 3456.19   158.1 3455.04   167.4 3452.88   190.2 3452.54
   202.2 3453.59   206.6 3454.41   219.6 3455.13   231.2 3453.18   246.5 3452.62
   264.4 3453.22   271.1 3456.26   275.5  3457.3   327.1 3458.52   342.8 3462.17
   361.8 3464.58   399.3 3474.08   425.2 3481.75   454.1 3488.42   479.6 3492.73
#Mann= 4 ,-1,0
       0     .12       0     110      .1       0   231.2    .045       0
   264.4      .1       0
#XS Ineff= 2 , 0
           214.4 3458.18   281.2         3458.11
Permanent Ineff=
       F       F
Bank Sta=231.2,264.4
XS Rating Curve= 0 ,0
Exp/Cntr(USF)=0,0
Exp/Cntr=0.5,0.3

Type RM Length L Ch R = 1 ,84022   ,222.3,208.3,187.8
BEGIN DESCRIPTION:
structure xs 2
END DESCRIPTION:
XS GIS Cut Line= 5
2203488.47008832448914.0412854492203313.51379746448990.010892692
  2203256.440054448989.9709059952203134.82678664449046.518537269
2203020.21479813 449109.41536023
#Sta/Elev= 30
       0 3489.74    26.5 3484.97    39.6 3480.15    58.1 3480.18    87.5 3476.64
    91.9 3475.47     105 3469.65   126.8 3458.89   130.3 3457.96     179 3455.88
   247.8 3454.43   255.4 3453.08   274.4 3452.56  279.39 3453.05   283.5 3454.23
   305.5 3454.45   331.7 3457.04     354 3458.02   369.3 3460.67   387.5 3461.76
   400.6 3463.42   412.4 3466.72   424.1  3471.4     429 3472.89   438.9 3474.31
   448.8 3476.32   480.1 3484.51   489.9 3486.29   508.1 3490.93   512.7 3491.55
#Mann= 5 ,-1,0
       0      .1       0      50     .12       0     110      .1       0
   255.4    .045       0  279.39      .1       0
#XS Ineff= 2 , 0
           244.2 3457.57   290.6         3457.57
Permanent Ineff=
       F       F
Bank Sta=255.4,279.39
XS Rating Curve= 0 ,0
Exp/Cntr(USF)=0,0
Exp/Cntr=0.5,0.3

Type RM Length L Ch R = 1 ,83814   ,186.7,196.2,203.9
XS GIS Cut Line= 4
2203181.88292826448758.9014604182203111.99756942448842.763891034
2203042.11221057449002.7237123922202993.96896336449075.715087187
#Sta/Elev= 30
       0 3506.14    39.4 3495.04    75.9 3484.07    81.1 3482.14    93.7 3474.72
   101.9 3471.21   107.1 3468.17   111.8 3464.38   116.2 3459.92   120.5 3456.59
   124.9 3454.79   132.1 3453.26   150.4 3451.89   159.8 3453.27   172.9 3454.33
   183.8 3453.81   208.1 3453.65     234 3454.84   255.8 3454.66   268.9 3455.26
   273.3 3456.35   277.7 3458.07   294.5  3466.2     309 3471.85   310.6 3472.33
     325 3472.97   327.3 3473.43   344.6 3480.18   359.9 3484.26371.1628 3488.05
#Mann= 4 ,-1,0
       0      .1       0     100     .12       0   132.1    .045       0
   159.8      .1       0
Bank Sta=132.1,159.8
XS Rating Curve= 0 ,0
Exp/Cntr(USF)=0,0
Exp/Cntr=0.3,0.1

Type RM Length L Ch R = 1 ,83618   ,200.9,205.8,210.3
XS GIS Cut Line= 4
2203048.32424247448710.7582132132202984.65091552 448766.66650029
2202888.36442111448873.8240505212202855.75125365448993.405664546
#Sta/Elev= 30
       0 3491.68      16 3487.58    58.2 3478.66    64.2 3477.15    70.4 3474.81
    75.5 3472.37    81.2 3469.31    88.1 3465.11   103.8 3456.93   106.7 3455.94
     115 3454.54   125.8 3454.38   133.3 3453.25   137.8 3453.03     152 3453.21
     158 3452.78   169.2 3451.96   179.5 3452.13  192.223453.075     201  3453.8
   206.4 3454.89   217.1 3460.25   222.8 3462.01   232.3 3464.51     253 3468.56
   265.4 3471.39   290.3 3474.87   319.3 3480.24   340.1  3483.7352.7461 3486.36
#Mann= 4 ,-1,0
       0     .12       0      70      .1       0     158    .045       0
  192.22      .1       0
Bank Sta=158,192.22
XS Rating Curve= 0 ,0
Exp/Cntr(USF)=0,0
Exp/Cntr=0.3,0.1

Type RM Length L Ch R = 1 ,83412   ,325.3,311.2,293.8
XS GIS Cut Line= 4
2202916.31856465448581.8585513422202865.06930149448625.342774624
 2202731.5106157448726.2882929572202636.77712926448814.809747495
#Sta/Elev= 30
       0 3481.79      36  3476.5    42.2 3475.38    50.7 3473.13    54.6 3471.56
    67.7 3464.35    80.2 3455.47    83.4 3454.02    87.7 3452.87    96.3 3452.16
   107.7 3451.96   133.3 3452.46   144.8 3453.09   153.2 3452.63  157.323451.543
   163.6 3450.14  173.223451.544   193.7 3452.24   203.7 3454.62   208.7 3455.28
   244.7 3458.03   270.2    3459   278.7 3459.87   293.9 3459.81   315.8 3461.54
   326.8 3464.46   337.7 3468.92   343.2 3470.25   354.2 3474.17 364.282 3477.06
#Mann= 4 ,-1,0
       0     .12       0      20      .1       0  157.32    .045       0
  173.22      .1       0
Bank Sta=157.32,173.22
XS Rating Curve= 0 ,0
Exp/Cntr(USF)=0,0
Exp/Cntr=0.3,0.1

Type RM Length L Ch R = 1 ,83101   ,308.9,310.1,300.8
XS GIS Cut Line= 4
 2202850.7279439448075.1178011912202691.59255888448264.929886946
2202603.39704428448677.148052978 2202555.4646994448753.839804798
#Sta/Elev= 30
       0 3469.54    10.2 3467.87    28.8 3457.54    34.5 3455.49    60.1 3454.06
    70.5  3452.3    99.8 3453.95   122.7 3454.05   142.4 3455.76   169.7 3453.84
   190.8 3456.81   362.5  3452.6   391.1 3453.22     477  3451.8   501.6 3452.29
  515.423451.014   530.2 3448.22   534.3 3448.62  539.963451.015     567 3451.35
   583.4 3453.11   611.3 3452.83   636.5    3454   644.7 3455.59   661.1 3464.24
   683.4 3467.51   711.7  3468.9   725.9 3470.77   743.2  3475.3759.6808 3478.07
#Mann= 4 ,-1,0
       0     .12       0  327.69      .1       0  515.42    .045       0
  539.96      .1       0
#XS Ineff= 2 , 0
          190.31 3457.46
Permanent Ineff=
       F       F
Bank Sta=515.42,539.96
XS Rating Curve= 0 ,0
Exp/Cntr(USF)=0,0
Exp/Cntr=0.3,0.1

Type RM Length L Ch R = 1 ,82791   ,626.4,653.8,649.4
XS GIS Cut Line= 4
2202417.41954612448000.3433431672202398.24660816 448224.66671724
2202363.73531984448571.6968942262202342.64508809448671.396171592
#Sta/Elev= 30
       0 3470.71    20.9 3469.57      57 3463.58   101.2 3462.12   173.5 3461.38
   192.7 3460.26   205.6 3458.66   217.6 3459.38   229.7 3457.75   245.7 3453.32
   249.8 3452.87   322.6 3451.26   358.3 3451.69   394.5 3451.12   398.5 3449.73
   402.5 3447.75   406.5 3447.63   414.6 3447.97   418.6 3449.67   430.7 3450.66
     495 3450.45   527.1 3451.19   551.3  3453.4   571.4 3457.16   591.8 3464.86
     604 3470.54   612.2 3472.57   624.5 3476.89   640.8 3480.88675.7888 3486.35
#Mann= 4 ,-1,0
       0     .12       0  245.14      .1       0   398.5    .045       0
   418.6      .1       0
Bank Sta=398.5,418.6
XS Rating Curve= 0 ,0
Exp/Cntr(USF)=0,0
Exp/Cntr=0.3,0.1

Type RM Length L Ch R = 1 ,82137   ,280.7,281.8,281.1
XS GIS Cut Line= 4
2202032.04349322448092.3734453512202033.96078702448261.095299355
 2202041.6299622448558.2758376572202049.29913738448636.884883273
#Sta/Elev= 30
       0 3467.46   116.8 3461.97   168.8 3460.23   176.8 3458.89   192.8 3452.88
   200.8 3450.97   212.8 3450.16   224.8 3450.43   240.8 3448.47   248.8 3447.39
   256.8    3447   264.6 3448.35   276.9 3449.23   284.9 3448.96   292.9 3449.49
   328.9 3449.56   356.9 3448.99   368.9 3449.62   408.9 3449.69   425.3 3450.18
   444.9 3451.64   448.9 3452.48   468.9 3468.16   472.9 3470.82     477 3472.55
     481 3473.45   497.1 3473.74   501.1 3474.25   521.2 3479.15544.9945 3482.79
#Mann= 4 ,-1,0
       0      .1       0      60     .12       0   240.8    .045       0
   264.6      .1       0
Bank Sta=240.8,264.6
XS Rating Curve= 0 ,0
Exp/Cntr(USF)=0,0
Exp/Cntr=0.3,0.1

Type RM Length L Ch R = 1 ,81855   ,388.8,391,379.6
XS GIS Cut Line= 4
2201778.96071222448117.2982646922201796.21635638448309.027644242
2201807.72011915 448587.035244592201813.47200054448659.892408819
#Sta/Elev= 30
       0 3475.93    37.9 3474.07    55.9 3471.77    80.2 3465.38   100.3 3462.84
   116.3 3456.64   144.5 3452.88   164.5 3456.15   184.6 3455.43   212.7 3451.29
   224.7 3451.32   236.7 3449.12   244.7 3448.51   268.7 3448.22   288.7 3449.12
   292.9 3448.62   296.7 3446.44   304.1 3445.73   308.8 3446.07   316.8 3448.73
   424.9 3449.36   444.9 3450.37   450.2  3452.6   460.9 3461.28   468.9 3464.73
   476.9 3466.58     501  3469.6     517 3473.11   525.1 3473.75543.8337 3478.41
#Mann= 7 ,-1,0
       0      .1       0      30     .12       0   232.5      .1       0
   292.9    .045       0   316.8      .1       0   422.5     .12       0
  520.75      .1       0
Bank Sta=292.9,316.8
XS Rating Curve= 0 ,0
Exp/Cntr(USF)=0,0
Exp/Cntr=0.3,0.1

Type RM Length L Ch R = 1 ,81464   ,600.2,600.2,600.2
XS GIS Cut Line= 4
 2201573.8102761448213.1629544672201594.90050785448322.448700811
2201646.66744033448581.2833632032201669.67496587448667.561584001
#Sta/Elev= 30
       0 3471.07    24.5 3469.79    29.4 3467.79    40.8 3460.94    44.8    3460
    69.3 3458.06   114.1 3457.02   124.9 3449.29   130.4 3448.17     159 3447.75
   191.6 3448.28   220.1 3447.66   244.6 3448.62   260.9 3447.75   273.2 3448.24
   277.3 3447.82   281.3 3446.28   285.4 3446.01   297.7 3446.29  301.98 3447.97
   305.8  3448.8   342.5 3449.31   368.1 3451.86   379.3 3453.51   396.6 3458.47
   408.3 3459.88   427.7 3458.65     432 3459.02   445.5 3461.61 464.556 3466.82
#Mann= 5 ,-1,0
       0      .1       0   231.3     .12       0   277.3    .045       0
  301.98     .12       0  435.26      .1       0
Bank Sta=277.3,301.98
XS Rating Curve= 0 ,0
Exp/Cntr(USF)=0,0
Exp/Cntr=0.3,0.1

Type RM Length L Ch R = 1 ,80864   ,304.3,310.5,304.3
XS GIS Cut Line= 4
2201303.47185093448332.0351697882201334.14855166448410.644215404
2201378.24630896448575.5314818172201414.67489107448700.155578524
#Sta/Elev= 30
       0 3474.31    16.9 3471.29    34.9 3467.44    44.2 3466.74      57 3464.62
    69.9 3459.56    74.2 3456.93    82.8 3450.44      87 3447.99    90.8 3446.65
    95.3 3445.04   120.1 3444.69   128.4 3446.52   137.1 3447.57   153.4 3447.09
     173 3447.62   189.4 3447.59   202.9 3447.07   223.6 3448.25   237.7 3448.51
   264.4 3448.49   296.6 3446.87   302.6 3446.95   306.8 3447.86   319.3    3452
   327.6 3455.62     336 3457.45   348.2 3461.58   361.1  3464.6384.9041 3468.26
#Mann= 3 ,-1,0
       0      .1       0    90.8    .045       0   128.4      .1       0
Bank Sta=90.8,128.4
XS Rating Curve= 0 ,0
Exp/Cntr(USF)=0,0
Exp/Cntr=0.3,0.1

Type RM Length L Ch R = 1 ,80553   ,305.6,308.2,307.8
XS GIS Cut Line= 4
2201134.74999693448491.1705548152201180.76504802448642.636764659
2201217.19363014 448761.50897998 2201232.5319805448811.358618663
#Sta/Elev= 30
       0 3476.25      23 3474.36    35.5  3472.6    46.2 3471.86      69 3467.75
    73.2 3466.23    77.3 3464.23    89.9  3454.8    94.1 3453.07   102.2 3450.94
   111.8 3447.71     115 3447.25     131 3447.37   144.2 3446.32   165.1 3447.02
   173.5 3446.18   181.9    3446   198.6 3446.79   202.8  3446.5     207 3445.59
   211.2 3444.69   227.9 3445.48   238.2 3446.38   259.1 3447.01   265.6 3447.57
   269.7 3448.93   278.3 3454.04   290.7 3459.56   307.4 3466.26334.7864  3472.4
#Mann= 3 ,-1,0
       0      .1       0     207    .045       0   227.9      .1       0
Bank Sta=207,227.9
XS Rating Curve= 0 ,0
Exp/Cntr(USF)=0,0
Exp/Cntr=0.3,0.1

Type RM Length L Ch R = 1 ,80245   ,308.1,306.6,300.3
XS GIS Cut Line= 4
2200879.74992213448611.9600639312200908.50932906448719.328516479
2200931.51685461448830.5315566182200948.77249877448909.140602234
#Sta/Elev= 30
       0 3479.07     9.5 3477.39      22 3475.81    34.4 3472.59    42.7 3469.71
    67.5  3462.3    71.7 3460.61    84.1 3454.46    88.2 3452.89    91.6 3451.95
  127.173446.367   137.6 3444.99   141.6 3445.76   149.8  3445.9   153.9 3446.27
   162.1 3446.32   182.5 3447.14   186.6 3447.09   198.8 3446.16   208.2 3446.42
   215.2 3447.21   243.1 3454.93   247.9 3456.41   256.1 3459.48   264.3 3461.55
   268.4 3463.08   280.7 3470.43   283.7 3471.29   290.3 3472.05305.1923 3472.09
#Mann= 3 ,-1,0
       0      .1       0  127.17    .045       0   153.9      .1       0
Bank Sta=127.17,153.9
XS Rating Curve= 0 ,0
Exp/Cntr(USF)=0,0
Exp/Cntr=0.3,0.1

Type RM Length L Ch R = 1 ,79939   ,214.1,209.3,203.2
XS GIS Cut Line= 4
2200607.49420317448717.4112226842200628.58443492 448799.85485589
2200672.68219221448926.3962463932200695.68971776448989.666941645
#Sta/Elev= 30
       0 3476.78       8 3475.71    12.1 3474.84    23.4 3471.98    28.7 3470.22
    36.9 3467.03    65.8 3453.01      76 3449.02    82.3 3447.16   110.9 3444.98
   133.1 3444.22   154.9 3444.39   170.6 3443.89   179.7 3442.79   188.2 3442.95
   191.9 3443.73   196.6 3445.43   198.9  3445.9   209.3 3446.71   213.6 3447.34
   222.1 3451.35   230.2 3456.94   234.8 3459.42   239.1 3460.29   247.6 3460.43
   255.2  3461.2   260.4 3463.05   264.6 3465.26   276.1 3467.45286.4275 3468.81
#Mann= 3 ,-1,0
       0      .1       0   170.6    .045       0   191.9      .1       0
Bank Sta=170.6,191.9
XS Rating Curve= 0 ,0
Exp/Cntr(USF)=0,0
Exp/Cntr=0.3,0.1

Type RM Length L Ch R = 1 ,79729   ,269.9,277.3,281.9
XS GIS Cut Line= 4
2200406.17835464448820.9450876412200457.94528712448899.554133256
 2200507.7949258448976.2458850762200544.22350791449056.772224487
#Sta/Elev= 30
       0 3468.45    43.4 3464.91    61.8 3458.37    73.8 3452.21    81.7  3449.2
    91.3 3447.44   105.6 3445.82  108.523444.662   111.4 3443.46   115.1 3442.41
   119.3 3442.38   124.7 3442.53   127.6 3442.92   129.5 3443.32  132.723444.662
   134.2 3445.29     139 3445.92   172.1 3446.39   177.2 3446.84   181.9 3448.33
   192.6  3453.5   199.8 3457.52   204.2 3459.18   225.3 3465.19     238 3467.91
     244 3470.31     247 3471.18   256.9 3471.71   258.9 3472.22273.9754 3477.93
#Mann= 3 ,-1,0
       0      .1       0  108.52    .045       0  132.72      .1       0
Bank Sta=108.52,132.72
XS Rating Curve= 0 ,0
Exp/Cntr(USF)=0,0
Exp/Cntr=0.3,0.1

Type RM Length L Ch R = 1 ,79452   ,389.9,387.4,382.1
XS GIS Cut Line= 4
2200178.02039297448901.4714270522200206.77979991448987.749647849
2200235.53920684449074.0278686472200268.13320136449160.306089444
#Sta/Elev= 30
       0 3462.89     8.1 3461.93    33.1 3460.71    45.7 3459.32    54.5 3457.74
    67.9 3456.51    75.6 3454.82    77.4 3454.16    79.8  3453.1      84    3450
    88.2  3447.4    92.5 3446.26   105.1 3444.25  119.133443.665   150.1 3442.37
   151.5 3442.37  154.853443.663   155.7 3443.98   164.1 3449.37   168.3 3451.58
   172.2 3454.08   181.7 3458.08   184.8 3459.22   187.9 3459.89   203.4 3461.95
   209.7 3462.11   223.7 3461.87   240.3 3462.42   270.8 3465.79274.1201 3465.92
#Mann= 4 ,-1,0
       0      .1       0  119.13    .045       0  154.85     .12       0
  211.89      .1       0
Bank Sta=119.13,154.85
XS Rating Curve= 0 ,0
Exp/Cntr(USF)=0,0
Exp/Cntr=0.3,0.1

Type RM Length L Ch R = 1 ,79065   ,326.3,327.7,326.9
XS GIS Cut Line= 4
2199800.31351526 449047.185755512199840.57668497 449106.62186317
2199898.09549883449208.238434332 2199955.6143127449319.441474471
#Sta/Elev= 30
       0 3469.25    12.9 3465.79    26.6 3460.83    38.8 3458.36    50.3 3454.85
    70.5 3446.97    79.3 3444.89    88.5 3443.93    93.1 3442.89   95.933441.795
    97.7 3441.12   102.3 3440.26   116.1 3440.19   120.3 3440.64  123.573441.797
   126.2 3442.57   139.1  3443.5   152.2 3443.07   161.4 3443.42   176.1 3446.89
     179 3447.23   189.6 3447.31   198.6 3446.16   210.5 3446.58   234.6 3450.99
   247.2 3452.94     254 3453.59   270.7    3454   291.7 3453.67313.7539 3454.87
#Mann= 4 ,-1,0
       0      .1       0   95.93    .045       0  123.57      .1       0
  208.56     .12       0
Bank Sta=95.93,123.57
XS Rating Curve= 0 ,0
Exp/Cntr(USF)=0,0
Exp/Cntr=0.3,0.1

Type RM Length L Ch R = 1 ,78737   ,541.9,563.5,557.3
XS GIS Cut Line= 4
2199543.39614666449198.6519653542199566.40367221449271.509129583
2199691.02776892449486.2460346792199792.64434008449549.516729931
#Sta/Elev= 30
       0 3462.37    19.4  3458.7    37.7 3453.75      53 3451.61    63.2 3449.58
    78.3  3444.7      83 3443.96    92.2 3441.44  110.783440.428   115.3 3439.61
     120 3439.28   129.2 3439.25   138.5 3439.51   145.33440.427   161.6 3443.22
   178.4 3443.22     196 3444.29   254.1  3443.4   263.3 3442.09     268 3442.07
   298.4 3443.14     316 3444.55   335.5 3445.33   345.1 3447.16   354.3 3449.69
   369.1 3453.12   396.7 3461.09   414.8 3465.58   426.4 3467.57444.3882 3469.89
#Mann= 4 ,-1,0
       0      .1       0  110.78    .045       0   145.3      .1       0
   256.4     .12       0
#XS Ineff= 2 , 0
                          198.79         3446.35
Permanent Ineff=
       F       F
Bank Sta=110.78,145.3
XS Rating Curve= 0 ,0
Exp/Cntr(USF)=0,0
Exp/Cntr=0.3,0.1

Type RM Length L Ch R = 1 ,78174   ,152,152.9,153.7
XS GIS Cut Line= 4
2199231.88699254449343.4382995062199282.01102776449512.438739624
2199460.95251346449693.4126078042199607.65527402449839.591036505
#Sta/Elev= 30
       0 3465.51    22.7 3460.64      31 3458.02    40.2  3453.5    51.9 3450.09
    56.1 3449.65   117.5 3447.73   133.6 3448.99   146.4 3447.63   196.4 3445.52
   213.5 3443.43   230.6  3442.6   305.6 3441.21   342.4 3441.37   357.3 3442.91
   370.7 3442.86   387.6  3442.2   401.2 3440.51   424.8 3441.68   449.9  3440.4
   466.8 3438.36   514.4 3437.54   531.9 3438.46   538.1  3441.3     546  3449.6
   555.1 3457.33   568.7 3464.66   600.5 3470.18   628.1 3476.11   637.9 3479.08
#Mann= 9 ,-1,0
       0     .12       0     110      .1       0  296.28     .12       0
  336.28      .1       0  430.78     .12       0   466.8    .045       0
   531.9      .1       0  570.78     .12       0  610.78      .1       0
#XS Ineff= 2 , 0
          362.69  3445.6
Permanent Ineff=
       F       F
Bank Sta=466.8,531.9
XS Rating Curve= 0 ,0
Exp/Cntr(USF)=0,0
Exp/Cntr=0.3,0.1

Type RM Length L Ch R = 1 ,78021   ,249.7,247.8,246.6
XS GIS Cut Line= 3
2199049.92799752449280.7686375892199157.89803042449657.565772432
2199528.81063922449930.885418047
#Sta/Elev= 30
       0 3465.05    12.9 3464.78    37.9 3458.84    50.4 3454.17    62.8 3453.16
      92 3454.93   183.3 3452.97   260.9 3449.84   279.2 3446.41   345.8 3447.31
   358.3 3448.56   374.9  3446.8   404.7 3446.66   439.5 3442.02   472.2    3444
   489.2 3442.92   499.1 3443.87     519 3442.75   628.3  3443.1   638.3 3442.48
   659.4 3437.54   673.7 3436.65     683 3437.57   737.6 3442.16   747.6 3446.29
   772.4 3463.69   822.1 3471.08     831 3473.94   845.3 3474.88   852.7 3477.22
#Mann= 6 ,-1,0
       0      .1       0      50     .12       0     260      .1       0
  651.96     .12       0   659.4    .045       0     683      .1       0
#XS Ineff= 2 , 0
          627.63 3444.77
Permanent Ineff=
       F       F
Bank Sta=659.4,683
XS Rating Curve= 0 ,0
Exp/Cntr(USF)=0,0
Exp/Cntr=0.3,0.1

Type RM Length L Ch R = 1 ,77773   ,99.3,100.1,100.4
XS GIS Cut Line= 4
2198956.70424524449217.8249033092199167.60656275449982.825127714
2199317.15547879450069.1033485112199411.10287477450128.539456172
#Sta/Elev= 30
       0 3466.83    28.4 3464.61    57.4 3457.67      74 3456.37   115.5 3457.67
   132.4 3456.39   151.9 3456.96     186 3454.22   264.9 3453.37     323 3449.68
   360.3 3449.02   397.7 3450.45   576.1 3446.07   625.9  3442.7   656.1 3443.74
   667.4  3442.8   679.8 3443.94   721.3  3443.3   863.5 3438.63  875.573436.941
   889.4 3435.47     905 3435.75  908.453436.941   928.1 3451.65   942.3 3458.88
   993.4 3466.12  1011.9 3471.29  1021.8 3471.77  1059.7 3486.041077.362 3490.15
#Mann= 7 ,-1,0
       0      .1       0      10     .12       0      40      .1       0
     120     .12       0     320      .1       0  875.57    .045       0
  908.45      .1       0
Bank Sta=875.57,908.45
XS Rating Curve= 0 ,0
Exp/Cntr(USF)=0,0
Exp/Cntr=0.3,0.1

Type RM Length L Ch R = 1 ,77673   ,228.4,237.3,242.8
XS GIS Cut Line= 4
2198807.15532919449865.8702061882199133.09527443450074.855229898
2199276.89230909450163.050744491 2199355.5013547450210.983089378
#Sta/Elev= 30
       0 3484.37    15.5 3483.33    29.7 3479.38    58.2 3474.87    72.5  3469.2
      82  3468.3   110.5 3461.88     139  3449.7   153.3 3444.96   181.8 3443.55
   300.6 3441.92     310 3440.61   333.8 3441.88   348.1 3440.49   357.6 3440.99
   402.7  3440.1   452.2 3437.76  463.413436.101   472.6 3434.87   489.3 3434.91
  493.943436.101   507.5 3443.04   521.7 3454.78   531.6 3460.24     560 3464.06
   580.2 3469.09   592.5 3469.82   601.9 3474.13   613.7 3477.47647.9434 3489.51
#Mann= 7 ,-1,0
       0     .06       0      80      .1       0     310     .12       0
  427.18      .1       0  463.41    .045       0  493.94     .12       0
  547.18      .1       0
#XS Ineff= 2 , 0
          400.88 3442.45
Permanent Ineff=
       F       F
Bank Sta=463.41,493.94
XS Rating Curve= 0 ,0
Exp/Cntr(USF)=0,0
Exp/Cntr=0.3,0.1

Type RM Length L Ch R = 1 ,77435   ,307.9,319,315.3
XS GIS Cut Line= 4
2198720.87710839449980.9078339182199019.97494049 450256.99814047
2199129.26068684 450368.201180612199194.44867588 450444.89293243
#Sta/Elev= 30
       0 3491.47     9.9 3485.61    37.1 3485.48    47.8 3480.39    91.6 3467.74
   113.4 3459.23   147.8 3438.94   152.6  3437.5     244 3436.26   265.8 3437.66
     293 3434.99   336.5 3433.56   354.2 3435.13   441.3 3436.52   455.4 3433.81
   464.4 3432.37   481.5 3433.85   506.3 3434.84   527.2 3433.72   531.8 3435.92
   544.3 3446.67   553.1 3451.86   565.7 3463.12   573.6 3468.44   591.3 3475.01
   602.6 3476.89   611.5 3481.08   636.7 3488.68   653.9 3495.39 663.613  3497.2
#Mann= 5 ,-1,0
       0     .06       0      70      .1       0     340     .12       0
   455.4    .045       0   481.5      .1       0
#XS Ineff= 2 , 0
          263.66 3440.82
Permanent Ineff=
       F       F
Bank Sta=455.4,481.5
XS Rating Curve= 0 ,0
Exp/Cntr(USF)=0,0
Exp/Cntr=0.3,0.1

Type RM Length L Ch R = 1 ,77116   ,165.1,165.4,163.6
XS GIS Cut Line= 4
2198605.83948066450187.9755638322198793.73427262 450427.63728827
2198857.00496787450527.3365656362198922.19295692450627.035843002
#Sta/Elev= 30
       0 3481.62     3.8 3480.16    13.9 3473.35    45.3 3461.25    62.5 3453.53
      93  3437.9   105.1 3434.28   116.5 3433.25   128.6 3433.91   143.8 3432.63
   194.7  3433.6   217.7 3432.95   230.3 3433.81   265.8 3431.46   276.1 3432.57
     296 3432.84   315.8 3432.41  325.743430.794   334.8 3429.76  368.093430.794
     377 3431.89   382.2 3433.58   398.7    3448   410.6 3453.31   472.5 3460.78
   486.9 3464.06   495.6 3467.15     510 3467.66     530  3475.1541.7364 3480.54
#Mann= 4 ,-1,0
       0     .06       0     110      .1       0  325.74    .045       0
  368.09      .1       0
#XS Ineff= 2 , 0
          192.98 3435.53
Permanent Ineff=
       F       F
Bank Sta=325.74,368.09
XS Rating Curve= 0 ,0
Exp/Cntr(USF)=0,0
Exp/Cntr=0.3,0.1

Type RM Length L Ch R = 1 ,76951   ,415.5,434.6,444.4
XS GIS Cut Line= 2
2198480.27537116450287.9933855982198814.36963402450716.909261765
#Sta/Elev= 30
       0 3484.82     6.5 3480.54    11.6 3478.58    32.1 3478.18    42.1 3473.37
    94.8 3455.52     104 3453.37   123.2 3443.47   136.5 3435.11   148.5 3430.66
     186 3430.11   199.2 3431.56   208.1 3430.86   273.2 3432.21   300.6 3429.82
   317.1 3428.85   331.1 3429.83   346.3 3431.61   371.3 3429.36   382.7    3431
   407.1 3429.81     414  3430.4   437.5  3439.1   456.8 3443.91     468 3451.47
     475 3454.28   493.3 3459.01   513.6 3462.51   525.2 3463.43   543.7 3470.69
#Mann= 4 ,-1,0
       0     .06       0     150      .1       0   300.6    .045       0
   331.1      .1       0
Bank Sta=300.6,331.1
XS Rating Curve= 0 ,0
Exp/Cntr(USF)=0,0
Exp/Cntr=0.3,0.1

Type RM Length L Ch R = 1 ,76516   ,225.4,204.6,186.4
XS GIS Cut Line= 4
 2198221.5101423450547.1101292332198380.01013616450798.697421079
2198388.81569137450864.1101169592198471.83949768450981.098207667
#Sta/Elev= 30
       0 3467.36     6.3 3466.32      15 3461.46    20.8  3459.3    35.3 3456.08
    52.7 3450.41    68.6  3446.2    82.8 3440.46    99.1 3428.71     102 3427.02
   104.9 3426.53   119.4 3426.02   142.7 3427.44   153.7 3426.99   160.1 3427.58
   189.1 3426.43   261.6 3427.19   299.9    3427  314.46 3426.19   335.3 3425.04
   340.2 3425.24  346.043426.284   364.7 3430.12   380.9 3438.48   389.2 3443.69
     399 3447.16   433.3  3453.3     453 3455.58   497.1 3462.35506.8094 3464.51
#Mann= 4 ,-1,0
       0     .06       0     110      .1       0  314.46    .045       0
  346.04      .1       0
Bank Sta=314.46,346.04
XS Rating Curve= 0 ,0
Exp/Cntr(USF)=0,0
Exp/Cntr=0.3,0.1

Type RM Length L Ch R = 1 ,76312   ,227.3,233.4,233.7
XS GIS Cut Line= 4
2198026.52999112450752.1537720872198220.25220584 450959.71328786
2198300.76013923451022.6101108222198380.01013616451079.217251487
#Sta/Elev= 30
       0  3447.3    34.2 3440.42      50 3436.32    72.6 3429.24    83.5  3427.2
    96.2 3422.74   109.4 3422.05   125.5 3424.56   132.7 3423.24   140.6 3422.95
   149.1 3421.35     166 3424.73   185.8 3423.37   194.3 3421.91   209.3 3424.01
     231 3425.34   247.6  3424.8     294 3425.58   304.9 3423.11   309.2 3422.53
   334.6 3422.46  353.533423.017   356.1 3424.17   380.3 3442.28   387.5 3445.35
   400.1 3448.49   421.9 3451.64   444.4 3456.11   467.8 3463.21483.4726 3464.46
#Mann= 5 ,-1,0
       0     .06       0      80     .12       0     230      .1       0
   304.9    .045       0  353.53      .1       0
Bank Sta=304.9,353.53
XS Rating Curve= 0 ,0
Exp/Cntr(USF)=0,0
Exp/Cntr=0.3,0.1

Type RM Length L Ch R = 1 ,76078   ,270.3,274.2,275.3
XS GIS Cut Line= 4
2197923.37920146450842.7251971522198115.84347972451130.792646315
2198157.35538288451193.6894692772198218.99426938451274.197402667
#Sta/Elev= 30
       0 3442.59    15.8 3440.24    28.3 3439.82    51.4 3435.42    73.4 3435.15
      86  3433.9     109 3429.85   120.6 3426.14   132.1 3420.84   149.4 3419.94
   158.1 3421.33   176.1 3420.44   195.8 3421.43   212.9 3420.77   238.8 3422.71
   257.9 3422.16   267.8 3422.75   301.2 3420.12   331.1 3421.88     347 3421.66
   367.8 3422.75   385.9 3421.31   397.2 3420.82     402 3421.32   414.8 3425.33
   431.2 3435.82   449.1    3441   465.9 3448.95   501.8 3457.77523.2022 3461.66
#Mann= 6 ,-1,0
       0     .07       0      70      .1       0     110     .12       0
     310      .1       0   385.9    .045       0     402      .1       0
Bank Sta=385.9,402
XS Rating Curve= 0 ,0
Exp/Cntr(USF)=0,0
Exp/Cntr=0.3,0.1

Type RM Length L Ch R = 1 ,75804   ,347.8,356.4,357.7
XS GIS Cut Line= 4
2197763.62127114450932.0386857572197890.67285352451116.955345264
2197974.95459629451241.4910547272198055.46252968451343.383907925
#Sta/Elev= 30
       0 3447.11    20.8 3442.21    45.1 3440.63    84.6 3434.06   103.3 3431.93
   122.7 3424.53   133.5 3422.58   142.1 3420.07   149.3 3419.12   161.5 3419.28
   171.2 3418.43   190.7 3418.71   208.3 3420.51   239.1 3421.66   253.6 3420.83
  257.06 3419.29   262.7 3418.62   268.1 3419.23   292.2 3419.89   319.8  3419.6
   329.3 3418.34   362.6 3420.53   389.6 3420.62   396.1 3419.27     410 3418.41
   449.4  3419.2   455.1  3421.2   479.9 3437.32   491.6 3442.19504.5924 3446.51
#Mann= 5 ,-1,0
       0      .1       0      40     .08       0      80      .1       0
  257.06    .045       0   268.1      .1       0
Bank Sta=257.06,268.1
XS Rating Curve= 0 ,0
Exp/Cntr(USF)=0,0
Exp/Cntr=0.3,0.1

Type RM Length L Ch R = 1 ,75448   ,433.7,443.8,444.2
XS GIS Cut Line= 4
2197518.32366159451076.7013785682197757.33158884451379.864065243
2197869.28793371451523.268821595 2197915.8315827451576.102152882
#Sta/Elev= 30
       0 3444.13    38.7 3435.44    67.6 3431.58    81.4 3427.42    95.6 3418.83
   104.2 3416.18   118.4 3417.76   151.6 3415.71   204.4 3414.73   216.2 3417.26
   229.1 3415.26   270.6 3415.63   290.9 3414.52   341.9 3417.32   364.8 3415.45
   371.9 3416.83   397.2 3418.01   423.2    3416   443.2 3416.83   448.6  3415.2
     474  3415.2   501.2  3416.9   514.2 3415.94   528.6 3416.57     540 3423.68
   554.3 3438.58     560 3442.35   594.1 3450.83   618.5 3458.96638.3896 3466.56
#Mann= 4 ,-1,0
       0     .06       0     120      .1       0   448.6    .045       0
     474      .1       0
Bank Sta=448.6,474
XS Rating Curve= 0 ,0
Exp/Cntr(USF)=0,0
Exp/Cntr=0.3,0.1

Type RM Length L Ch R = 1 ,75004   ,508.9,505.8,491.6
XS GIS Cut Line= 4
2197280.57367079451208.7847067882197398.81969796451446.534697582
2197504.48636054451708.1854811012197564.86731058451833.979127024
#Sta/Elev= 30
       0 3451.08       6  3450.3    26.1 3441.96    79.9 3429.36   101.4 3426.44
   147.9 3424.19   161.3 3421.23   174.7 3414.68     179 3413.92   250.6 3413.53
   285.6 3410.14   315.8 3412.77   339.3 3412.41   354.6 3409.59   367.6 3408.91
   403.8 3411.73   437.6 3411.07   459.1 3411.28   475.4 3412.74   505.6 3411.62
   556.2  3414.1   579.9 3412.67   605.2 3416.05   615.4 3420.77   632.2 3432.77
   641.2 3440.53   659.1 3458.67   664.2 3462.58   677.5 3470.27687.2483 3472.63
#Mann= 9 ,-1,0
       0     .06       0     100      .1       0     210     .12       0
     250      .1       0  315.53     .12       0  425.53      .1       0
   437.6    .045       0   459.1      .1       0  637.71     .08       0
#XS Ineff= 2 , 0
          192.73 3417.94  555.84         3417.33
Permanent Ineff=
       F       F
Bank Sta=437.6,459.1
XS Rating Curve= 0 ,0
Exp/Cntr(USF)=0,0
Exp/Cntr=0.3,0.1

Type RM Length L Ch R = 1 ,74498   ,269.6,267.4,263.3
XS GIS Cut Line= 4
2196967.34749245451464.1458080112197057.91891751451601.260882067
2197161.06970717451768.5664311442197225.22446659451884.296585393
#Sta/Elev= 30
       0 3436.07    15.6 3433.45   102.4 3421.87   116.8  3418.5     137 3410.13
   145.1 3408.25   164.2 3408.97   176.2 3407.07   211.2 3407.48   229.6 3405.76
   244.1 3406.37   250.2 3405.99   267.5 3404.75   276.4 3405.01   281.53406.114
   290.6 3407.35   314.2 3408.53   333.4 3407.65   363.6 3409.24     389 3408.46
   398.2 3409.15   402.7 3410.62   411.9 3415.79   434.2 3434.03   443.1 3437.68
     453 3444.34   457.8 3446.73   466.8 3453.14   481.3 3464.92493.1991 3472.17
#Mann= 7 ,-1,0
       0     .08       0      40      .1       0   250.2    .045       0
   281.5      .1       0  380.88     .08       0  430.88      .1       0
   493.2     .08       0
Bank Sta=250.2,281.5
XS Rating Curve= 0 ,0
Exp/Cntr(USF)=0,0
Exp/Cntr=0.3,0.1
