HEC-RAS study WILLIAMSRV.prj: WILLIAMSRV

--- WILLIAMSRV.g01 (geometry) --- (continued)

Type RM Length L Ch R = 1 ,74231   ,313.4,308.5,303.1
XS GIS Cut Line= 4
2196739.66099333451640.2569123032196864.19670279451781.145795737
2196943.44669972451876.7489666382197039.04987062452010.090231316
#Sta/Elev= 30
       0 3429.37     6.7 3426.49    11.9 3425.52      37 3423.29    63.4 3419.86
      76 3419.91   100.2 3418.16   121.6  3414.4   166.7 3410.58   193.7 3406.49
   213.1 3405.35  220.723403.859   227.8 3402.21     240 3402.03   245.2 3402.12
   249.2 3403.57   250.7 3404.21   263.2 3405.48   284.6 3404.23   304.5  3406.9
   341.7 3406.77   347.2 3406.18     357 3403.21   373.2 3404.58   381.7 3407.91
   401.3 3420.06   411.2    3424   430.2 3435.71   450.6 3449.86476.2916 3461.85
#Mann= 4 ,-1,0
       0     .06       0     100      .1       0  220.72    .045       0
   249.2      .1       0
#XS Ineff= 2 , 0
                          329.58         3410.38
Permanent Ineff=
       F       F
Bank Sta=220.72,249.2
XS Rating Curve= 0 ,0
Exp/Cntr(USF)=0,0
Exp/Cntr=0.3,0.1

Type RM Length L Ch R = 1 ,73922   ,368.7,365.8,355.8
XS GIS Cut Line= 4
2196527.69227701451872.5073375742196635.06072956451974.123908736
2196740.51188831452064.2367171242196867.05327882452179.274344855
#Sta/Elev= 30
       0 3431.75     6.8  3427.4    11.7 3425.84    23.5  3426.2    31.9 3425.52
    37.6 3424.11    50.2 3419.57    55.7 3418.41    74.4 3416.25    94.3 3412.76
   116.3 3410.17   145.1 3404.22   162.1 3402.95  172.293400.716   196.7 3400.16
   213.2 3400.68   257.2 3402.95     287 3402.65   296.9 3401.42   352.1 3399.57
   359.3 3400.03   366.3 3402.68   372.6 3406.32     395 3421.24   400.9 3425.82
   415.8 3442.97   422.9 3447.57   442.7  3454.3   448.4 3455.62457.5557  3456.2
#Mann= 4 ,-1,0
       0     .06       0     110      .1       0  172.29    .045       0
   213.2      .1       0
Bank Sta=172.29,213.2
XS Rating Curve= 0 ,0
Exp/Cntr(USF)=0,0
Exp/Cntr=0.3,0.1

Type RM Length L Ch R = 1 ,73556   ,352.2,323.4,292.3
XS GIS Cut Line= 4
 2196318.7072533452215.702926969 2196445.2486438452278.973622221
2196640.81261095  452372.92101822196775.02317663452365.251843018
#Sta/Elev= 30
       0 3433.21     6.1 3432.23    17.1 3425.74      24 3423.29     100 3412.52
   122.4 3409.57   140.3 3405.73   162.5 3397.41   175.3 3398.07  182.193397.063
   189.1 3396.51   205.3 3396.81   238.2 3399.33   264.5 3399.97   286.7 3399.29
   304.5 3397.67   331.2 3399.06   340.2 3398.08   373.8 3398.11   377.8 3397.82
   385.8 3395.64   397.9 3395.17   405.9 3395.37   409.9 3396.51   421.9 3408.03
   430.3 3410.16     454 3418.36     478 3423.83     486 3427.17492.8665 3428.68
#Mann= 4 ,-1,0
       0     .06       0     100      .1       0  182.19    .045       0
   205.3      .1       0
Bank Sta=182.19,205.3
XS Rating Curve= 0 ,0
Exp/Cntr(USF)=0,0
Exp/Cntr=0.3,0.1

Type RM Length L Ch R = 1 ,73233   ,361.7,362.5,362.3
XS GIS Cut Line= 4
2196401.15088651452741.041426936 2196489.3464011452660.515087525
2196652.31637372452486.0413521352196776.94047043452420.853363088
#Sta/Elev= 30
       0 3483.57    24.7 3471.89      36 3461.83    44.5 3456.12    47.3 3454.95
    65.1 3455.19    72.8 3452.48    82.8 3443.82    96.2 3434.17   112.4  3420.1
   132.3 3401.33   140.8 3395.96   151.4 3393.78   171.9 3393.83   184.2 3393.01
     203 3393.82   223.2 3395.19   260.8 3394.12   279.4 3396.79   322.8 3397.32
     336 3395.41   350.2 3396.88   376.1 3396.74   385.1 3394.21   394.3 3393.79
   407.7 3396.26   416.7 3396.27   429.8 3399.95   447.6 3400.45498.8186 3417.09
#Mann= 4 ,-1,0
       0     .06       0     110      .1       0   171.9    .045       0
     203      .1       0
#XS Ineff= 2 , 0
                          319.93         3401.45
Permanent Ineff=
       F       F
Bank Sta=171.9,203
XS Rating Curve= 0 ,0
Exp/Cntr(USF)=0,0
Exp/Cntr=0.3,0.1

Type RM Length L Ch R = 1 ,72871   ,188.4,192.2,194.6
XS GIS Cut Line= 4
2196698.33142481452967.2820948062196767.35400145452892.507636781
2196913.06832991452733.3722517542197010.85031348 452620.25191782
#Sta/Elev= 30
       0 3444.75     8.5 3439.53    20.4 3440.14    30.1 3438.97    50.9 3425.73
    73.6 3413.27    93.4 3405.03   114.8 3400.89   127.3 3392.44   143.43389.759
   155.7 3388.35  192.073389.759   209.5 3392.16   220.8 3392.12   241.9 3390.24
   258.1 3390.57   277.4 3392.32   301.5  3392.3   305.7  3392.7     317 3395.81
   351.1 3394.62   365.4 3395.09   387.9 3401.75   397.1 3403.64   410.6 3408.05
   423.5 3409.51   432.4 3413.58   444.7 3417.81     456 3423.27467.0556 3426.76
#Mann= 5 ,-1,0
       0      .1       0      10     .06       0  141.76      .1       0
   143.4    .045       0  192.07      .1       0
#XS Ineff= 2 , 0
                          280.84         3395.91
Permanent Ineff=
       F       F
Bank Sta=143.4,192.07
XS Rating Curve= 0 ,0
Exp/Cntr(USF)=0,0
Exp/Cntr=0.3,0.1

Type RM Length L Ch R = 1 ,72678   ,127.1,150.7,173.9
XS GIS Cut Line= 4
2196738.59459452453093.8234853092196845.96304707453065.064078376
  2197043.444308452892.5076367812197146.97817296452695.026375844
#Sta/Elev= 30
       0 3441.68     5.8 3433.59     9.9 3430.88    14.1 3429.87    30.6 3430.26
    34.8 3429.59    47.2  3423.1    67.9 3407.84    84.5 3397.55    96.9 3393.01
   119.4 3389.44   135.3 3388.22   172.5 3389.79  232.593388.051   252.2 3386.28
  272.173388.052   282.7 3391.23   287.3 3391.71   325.3 3390.68   376.4 3393.06
   395.2  3395.1   431.4  3396.6   449.4 3395.88   469.7 3398.05     481 3397.76
   517.2 3406.05   545.3 3408.93   566.8 3412.68   584.9 3413.36596.3781 3415.19
#Mann= 4 ,-1,0
       0     .06       0      70      .1       0  232.59    .045       0
  272.17      .1       0
#XS Ineff= 2 , 0
                          290.75         3393.79
Permanent Ineff=
       F       F
Bank Sta=232.59,272.17
XS Rating Curve= 0 ,0
Exp/Cntr(USF)=0,0
Exp/Cntr=0.3,0.1

Type RM Length L Ch R = 1 ,72528   ,214.2,217.6,225.2
XS GIS Cut Line= 4
2196745.25767851453109.3207996112196811.60841186453109.320799611
2197026.74563815453119.3739410272197290.13794324 453197.78844407
#Sta/Elev= 30
       0 3431.58     2.9 3429.52    18.9 3429.02    22.9 3428.45    26.9 3426.56
    54.9 3407.44    63.1  3403.2    74.9 3395.35    86.9 3389.39     115 3388.76
     131 3387.13     183 3389.06   191.1  3388.7   196.8 3387.24   203.1 3386.14
   242.7  3386.1  249.37 3387.09   267.1 3390.45   279.1  3391.6   312.4 3391.45
   354.2    3390   404.2  3391.1   438.7 3388.43   458.5 3388.81   466.8 3391.95
   483.2 3401.79   496.1 3412.57   516.9 3425.27   528.7 3430.22   556.5 3439.23
#Mann= 4 ,-1,0
       0     .06       0      60      .1       0   196.8    .045       0
  249.37      .1       0
#XS Ineff= 2 , 0
                          277.53         3393.36
Permanent Ineff=
       F       F
Bank Sta=196.8,249.37
XS Rating Curve= 0 ,0
Exp/Cntr(USF)=0,0
Exp/Cntr=0.3,0.1

Type RM Length L Ch R = 1 ,72310   ,234.2,234.6,238.9
XS GIS Cut Line= 4
 2196746.2637697453252.9588703352196926.48938648453312.394977996
2197047.27889559453350.7408539062197237.09098135453398.673198794
#Sta/Elev= 30
       0 3422.26     6.2  3418.8    20.7 3407.22    44.1 3390.16    48.3 3387.98
    51.8 3387.33    64.6 3387.06    73.6 3385.33   106.2 3386.77     122 3384.37
     141 3386.06   156.9 3385.85   175.9 3386.93   204.5 3386.43   217.2 3387.13
   233.5  3386.5   242.7 3384.45   262.9 3383.07  277.873384.633   296.5 3390.43
   304.9 3392.31   317.4 3393.15   321.6 3392.77   346.3 3394.86   358.8 3396.35
   391.7 3402.03   445.3 3416.24   465.9 3422.41   490.7 3431.84 512.274 3441.77
#Mann= 4 ,-1,0
       0     .06       0      60      .1       0   242.7    .045       0
  277.87      .1       0
Bank Sta=242.7,277.87
XS Rating Curve= 0 ,0
Exp/Cntr(USF)=0,0
Exp/Cntr=0.3,0.1

Type RM Length L Ch R = 1 ,72076   ,314.1,316.8,320.6
XS GIS Cut Line= 4
2196665.73743029 453383.334848432196719.42165656453419.763430544
2196955.24879341453552.0567024342197112.46688464453628.748454254
#Sta/Elev= 30
       0 3440.76    17.4 3422.65    22.3 3419.08    27.1 3416.98    41.6 3416.66
    46.5  3414.7    70.3 3397.27    97.8 3382.97     107 3382.31     130 3385.26
   148.7 3385.26   157.5 3384.42   162.1  3382.7   166.6 3381.67   198.6  3381.4
   209.4 3382.65   213.4 3383.67   230.9 3384.57     264 3384.12     278  3382.4
   281.3  3383.5   290.5  3389.6   295.6 3392.04   378.7 3407.13   392.6 3410.58
   417.6 3420.25   429.8 3423.31     452  3432.3   498.3 3448.79510.2029 3451.41
#Mann= 3 ,-1,0
       0     .06       0   162.1    .045       0   209.4      .1       0
Bank Sta=162.1,209.4
XS Rating Curve= 0 ,0
Exp/Cntr(USF)=0,0
Exp/Cntr=0.3,0.1

Type RM Length L Ch R = 1 ,71759   ,484.1,503.2,518
XS GIS Cut Line= 4
2196487.42910731453594.237165935 2196575.6246219453665.177036368
2196755.85023868453808.9740710312196880.47433539453904.838760806
#Sta/Elev= 30
       0 3414.43    11.2 3407.45    31.8 3407.12    36.8 3404.91    47.2 3397.65
    55.8 3394.48    76.6 3390.42   122.1 3384.29   133.5 3380.05   165.1 3380.46
   195.8 3383.03   216.2 3382.57   228.6 3381.02   246.9 3380.99   258.7 3378.82
   268.6 3378.44   292.8 3377.41  302.17 3378.45   313.5 3381.42   328.8 3391.36
   338.4 3399.27   344.1 3402.68   354.3 3404.78   370.3 3411.27   383.4 3414.35
   419.9 3429.35   429.7 3434.22     440 3436.79   460.2 3445.84500.9771 3460.87
#Mann= 5 ,-1,0
       0      .1       0      30     .07       0     100      .1       0
   268.6    .045       0  302.17      .1       0
#XS Ineff= 2 , 0
           199.1 3387.89
Permanent Ineff=
       F       F
Bank Sta=268.6,302.17
XS Rating Curve= 0 ,0
Exp/Cntr(USF)=0,0
Exp/Cntr=0.3,0.1

Type RM Length L Ch R = 1 ,71256   ,397.1,397,393.6
XS GIS Cut Line= 4
2196176.82751244453784.0492516892196295.69972776454006.455331968
2196358.97042301454152.169660426 2196404.9854741454240.365175019
#Sta/Elev= 30
       0 3413.06      21 3402.39      24 3401.51    42.1  3402.3    46.6 3400.75
    55.7 3395.74    73.8 3391.22    96.5  3381.9   110.1 3379.08   128.3 3377.88
   148.1 3380.32   168.3 3380.42   187.2 3379.21   246.2  3381.8   266.8 3379.45
     282 3375.51   303.1 3375.35  314.383373.929   320.6 3372.75   327.6 3372.66
  370.76 3373.93   381.6 3377.04     386 3379.36   394.5 3386.11   409.7 3401.97
   415.6 3406.81   425.7 3412.86   452.8 3424.39   497.9    3437510.5164 3439.36
#Mann= 4 ,-1,0
       0     .06       0      80      .1       0  314.38    .045       0
  370.76      .1       0
#XS Ineff= 2 , 0
          245.15 3384.11
Permanent Ineff=
       F       F
Bank Sta=314.38,370.76
XS Rating Curve= 0 ,0
Exp/Cntr(USF)=0,0
Exp/Cntr=0.3,0.1

Type RM Length L Ch R = 1 ,70859   ,301.3,303.3,305.9
XS GIS Cut Line= 3
2195781.18357277453901.6282138952196061.27735966454391.951533784
2196250.83511652454419.261449603
#Sta/Elev= 30
       0 3469.64    22.4 3459.39    30.2 3458.42    40.9 3453.45    50.2 3451.54
   100.8 3434.97   110.9 3430.59   127.9 3419.99   142.3 3420.11   146.9 3419.02
   159.3 3412.53   197.6 3398.46   252.8 3387.22   271.3 3378.81   291.6 3372.43
   300.9  3371.8   318.5  3373.8   333.2  3371.3     342 3370.06  371.86  3371.3
   412.3 3375.44   427.9 3374.34   441.7 3375.35   494.4 3374.48   506.2 3378.58
   567.6  3387.8   616.1 3401.64   684.8 3416.07   696.9 3418.12   756.2  3423.2
#Mann= 5 ,-1,0
       0      .1       0     170     .07       0     270      .1       0
   333.2    .045       0  371.86      .1       0
#XS Ineff= 2 , 0
                          412.85          3379.6
Permanent Ineff=
       F       F
Bank Sta=333.2,371.86
XS Rating Curve= 0 ,0
Exp/Cntr(USF)=0,0
Exp/Cntr=0.3,0.1

Type RM Length L Ch R = 1 ,70555   ,409.1,396.1,381.4
XS GIS Cut Line= 3
2195534.12146762454019.3134166492195758.41834587454499.260500212
2196069.53982215 454723.55737846
#Sta/Elev= 30
       0 3462.93    10.9 3457.94      30 3451.38   108.3 3426.06   125.7 3416.91
   143.3 3416.84   147.8  3415.2   152.2 3412.13   165.4  3407.4   231.7 3393.34
   240.7 3389.87   249.3 3384.81   252.7 3381.82   261.7 3374.86   271.4 3369.43
   275.8 3368.86   289.1 3370.42  318.05 3368.99   324.4 3367.35   337.6 3367.17
   346.4 3367.24     352 3368.93     361 3370.09   386.2 3371.95   442.3 3373.62
   694.7 3379.07   786.1 3386.27   830.4 3388.37   881.9 3388.66   913.3 3391.57
#Mann= 7 ,-1,0
       0      .1       0   152.2     .06       0   252.7      .1       0
  318.05    .045       0     352      .1       0     361     .12       0
   442.3      .1       0
Bank Sta=318.05,352
XS Rating Curve= 0 ,0
Exp/Cntr(USF)=0,0
Exp/Cntr=0.3,0.1

Type RM Length L Ch R = 1 ,70159   ,469.4,476.7,478.8
XS GIS Cut Line= 4
2195162.63845437454223.6215859862195300.67877786454469.322555783
2195944.04243501454899.0323716932196168.24077114454953.105403188
#Sta/Elev= 30
       0 3455.43    52.3 3434.24    79.8 3424.84   128.6 3403.71   149.2 3403.75
   166.5 3397.35   231.4  3387.1   248.1 3383.26   260.8    3376   272.5 3373.42
     286 3372.09   310.4 3374.19   339.2 3379.75   353.5 3375.32     363 3368.93
  389.61 3365.99   408.2 3364.62   425.4 3365.98   497.7 3367.56   728.6    3377
   762.2 3377.96   791.1 3376.63   922.5 3383.54  1031.6 3391.93  1146.2 3395.54
  1179.1 3398.99    1212 3398.14  1257.3 3400.18  1275.1  3402.9  1286.1 3403.04
#Mann= 12 ,-1,0
       0      .1       0     140     .06       0  311.82      .1       0
  389.61    .045       0   425.4      .1       0  551.82     .12       0
  591.82      .1       0  671.82     .12       0  771.82      .1       0
 1021.82     .08       0 1135.49      .1       0 1215.49     .08       0
Bank Sta=389.61,425.4
XS Rating Curve= 0 ,0
Exp/Cntr(USF)=0,0
Exp/Cntr=0.3,0.1

Type RM Length L Ch R = 1 ,69683   ,300.3,313.6,306.2
XS GIS Cut Line= 4
2194886.03932827454625.4186847362195010.30546435454761.710575917
2195298.92358685455046.3201133842195563.49019914455371.015501197
#Sta/Elev= 30
       0 3405.24      15  3400.6    37.6 3400.05    48.4 3396.96    80.6 3391.14
     116 3387.11   165.6 3378.76   182.6 3374.01   199.5 3365.31   223.6 3362.53
   237.6 3359.38   264.6 3359.82   276.9 3361.51   299.4 3361.01     366 3363.08
   411.6  3360.6   434.3 3359.91   445.6 3361.03   459.7  3363.7   501.7 3363.85
   513.5 3367.46   530.5 3368.26   580.3 3367.04   723.5 3370.72   774.1 3370.23
   781.7 3372.93   805.9 3385.92   820.5 3392.42   903.1 3417.591008.616 3455.33
#Mann= 6 ,-1,0
       0      .1       0      20     .06       0     160      .1       0
   411.6    .045       0   445.6      .1       0  829.78     .08       0
Bank Sta=411.6,445.6
XS Rating Curve= 0 ,0
Exp/Cntr(USF)=0,0
Exp/Cntr=0.3,0.1

Type RM Length L Ch R = 1 ,69369   ,261.1,259.5,257.9
XS GIS Cut Line= 2
2194673.34724533454761.9729131012195328.12868639455467.122157318
#Sta/Elev= 30
       0 3406.85    12.8 3406.97    31.7  3401.1    53.5 3397.08   186.4 3377.29
   199.6 3373.69   222.7 3361.97   277.3 3362.51   318.4 3360.09   386.3 3361.03
   403.9 3357.61     426 3356.56   439.2 3356.06   448.6 3356.55   479.3 3359.58
   497.9    3359     512 3361.78   553.4 3361.72   577.5  3364.3   609.6 3362.38
   644.9 3362.27   686.7 3364.18   744.8 3361.07   768.6 3361.16   785.5 3366.56
   812.2 3380.22   828.6 3390.58     845 3397.88   937.8 3425.82   962.3 3434.88
#Mann= 4 ,-1,0
       0     .06       0      90      .1       0     426    .045       0
   448.6      .1       0
#XS Ineff= 2 , 0
          275.57 3363.85  581.97         3367.26
Permanent Ineff=
       F       F
Bank Sta=426,448.6
XS Rating Curve= 0 ,0
Exp/Cntr(USF)=0,0
Exp/Cntr=0.3,0.1

Type RM Length L Ch R = 1 ,69110   ,734.7,751.1,734
XS GIS Cut Line= 4
 2194497.2065799454881.9681269592194745.73885206 455178.60341953
 2195062.4170698455455.1957869272195162.63169567455591.487678108
#Sta/Elev= 30
       0 3414.17    14.6 3408.87    44.1 3402.59    73.1 3394.54   110.5 3389.86
   132.2 3388.64   176.4 3383.24   272.4  3377.7   302.5 3377.27   378.3 3371.49
   384.9 3369.85     399 3362.02   413.2 3359.17   421.7  3355.1   427.4  3354.5
   495.4 3358.67   554.9 3356.41   570.8 3355.22   594.7 3356.41   603.2 3359.39
   613.3 3359.46   658.5 3357.78   767.9 3357.45   777.9 3361.62   795.9 3376.02
   804.4 3380.81   839.7 3390.99   890.2 3409.11   918.9 3417.27976.6215 3437.31
#Mann= 8 ,-1,0
       0     .06       0      70      .1       0     220     .12       0
     370      .1       0  506.99     .12       0   554.9    .045       0
   594.7     .12       0  616.99      .1       0
#XS Ineff= 2 , 0
                          699.42         3361.79
Permanent Ineff=
       F       F
Bank Sta=554.9,594.7
XS Rating Curve= 0 ,0
Exp/Cntr(USF)=0,0
Exp/Cntr=0.3,0.1

Type RM Length L Ch R = 1 ,68359   ,748.5,749.4,749.6
XS GIS Cut Line= 2
2194112.39110797455367.3042275552194677.15557964455961.434704519
#Sta/Elev= 30
       0  3392.9    22.9 3387.19    29.5 3386.39    43.6 3381.94    63.3 3373.72
    83.2 3361.41    94.5 3357.95   307.4  3355.6   313.2  3355.7   326.5 3358.06
   343.5 3356.14   388.8 3353.44   429.3 3354.92   453.9 3353.79   510.5 3356.12
   530.3 3354.04     557 3353.07   569.9 3353.89   592.5 3352.81   612.3 3348.92
   626.5 3347.31   653.8 3347.59   661.5  3349.1   666.1 3351.85   686.9 3367.97
   690.6 3369.63   725.6 3377.09   748.6 3384.33   764.2 3388.22   819.7 3408.57
#Mann= 5 ,-1,0
       0     .06       0      50      .1       0     340     .12       0
   612.3    .045       0   661.5      .1       0
#XS Ineff= 2 , 0
          507.04 3358.64
Permanent Ineff=
       F       F
Bank Sta=612.3,661.5
XS Rating Curve= 0 ,0
Exp/Cntr(USF)=0,0
Exp/Cntr=0.3,0.1

Type RM Length L Ch R = 1 ,67609   ,553.4,544.7,536.6
XS GIS Cut Line= 4
2193691.48098792  455948.2517462 2193827.7728791456080.535052346
2194040.22788594456284.9728891182194336.86317851456653.762712314
#Sta/Elev= 30
       0 3468.69    12.1 3463.62    40.7 3444.34    62.3 3432.63    83.2 3413.07
   105.8  3411.2   127.7 3396.85   173.8 3381.76   208.2  3358.7   219.7    3349
  235.143343.428   255.7 3341.72  272.643343.427     284 3347.44   298.2 3348.46
   357.6 3349.57   373.7 3347.07   401.4 3348.53   419.8 3351.81   462.3 3351.29
   479.3 3354.51   495.3 3359.95   521.9 3358.78     574 3362.38     593 3361.84
     740 3376.68   797.4 3377.91   813.6 3382.77     869 3388.65958.0595 3401.99
#Mann= 8 ,-1,0
       0      .1       0      90     .07       0     100     .06       0
  219.93      .1       0  235.14    .045       0  272.64      .1       0
  524.77     .12       0  654.77      .1       0
#XS Ineff= 2 , 0
                          356.83          3352.3
Permanent Ineff=
       F       F
Bank Sta=235.14,272.64
XS Rating Curve= 0 ,0
Exp/Cntr(USF)=0,0
Exp/Cntr=0.3,0.1

Type RM Length L Ch R = 1 ,67064   ,396.9,451.1,490.2
XS GIS Cut Line= 5
2193475.01739604456417.2561952642193535.14617156456553.548086445
 2193711.2580236456644.8494303542194033.27828724456750.645871567
2194139.32927054456860.151020843
#Sta/Elev= 30
       0 3409.34    22.7 3396.56    67.6 3376.82    88.8 3366.34   135.4 3350.54
   163.6  3346.3   172.7 3340.01   177.2 3339.08   199.7 3338.94   222.2 3339.13
228.7179 3340.06   235.7  3341.6   259.2 3342.31   289.8 3340.92   316.8 3345.49
   389.5 3345.73   398.8 3346.88   415.7 3355.28   440.9 3356.42   591.9 3357.75
   613.6  3356.5   626.2 3352.78   630.4 3352.47   664.1 3351.32   689.8 3353.11
   707.7 3361.02   723.2 3370.12   759.5 3388.03   776.7 3393.32   838.7 3405.91
#Mann= 5 ,-1,0
       0      .1       0   172.7    .045       0228.7179      .1       0
  288.97     .12       0  547.34      .1       0
Bank Sta=172.7,228.7179
XS Rating Curve= 0 ,0
Exp/Cntr(USF)=0,0
Exp/Cntr=0.3,0.1

Type RM Length L Ch R = 1 ,66613   ,500.4,498.4,497.6
XS GIS Cut Line= 4
2193326.69974976456441.3077054732193338.72550486456757.985923217
2193282.60531438456930.3550797112193230.49370892457086.689896066
#Sta/Elev= 30
       0 3401.34    39.9 3386.31    79.9 3369.66     112 3355.95     132 3345.78
     148 3342.77     164 3345.48     184 3343.55     208 3344.56   221.1 3342.07
     244 3344.14   255.8 3340.93   268.1 3339.89   284.1 3341.25   328.7    3342
   366.5 3339.91   381.8 3337.62   404.4 3338.35  412.663336.741   442.1 3335.06
  456.153336.743   463.3 3341.38   484.3 3360.18   496.9 3366.78   530.7 3375.18
   577.1 3390.99   606.3 3405.93     615 3408.83   627.6 3416.89662.9728 3433.51
#Mann= 4 ,-1,0
       0     .06       0      70      .1       0  412.66    .045       0
  456.15      .1       0
#XS Ineff= 2 , 0
          327.64 3344.55
Permanent Ineff=
       F       F
Bank Sta=412.66,456.15
XS Rating Curve= 0 ,0
Exp/Cntr(USF)=0,0
Exp/Cntr=0.3,0.1

Type RM Length L Ch R = 1 ,66115   ,699.5,698.6,699.7
XS GIS Cut Line= 4
2192925.84124628456425.2733653342192893.77256601456553.548086445
2192849.67813062456721.9086579042192821.61803538457026.561120545
#Sta/Elev= 30
       0 3392.32       4 3391.44    16.4 3384.65    41.1 3376.05    86.5 3364.21
    98.9 3363.13   115.3 3360.14   132.2 3355.66   140.1 3351.93   160.8 3336.35
  178.863332.196   210.4 3330.83  219.793332.196   222.8 3332.98   247.9 3333.79
   276.6 3335.83     329 3334.73   357.7 3335.58   377.8 3334.55   385.9 3333.36
   389.9 3333.72     418 3343.44   440.9  3353.6   474.2 3366.58   498.2 3377.73
   526.5 3387.62   534.5 3391.52   570.6 3406.53   594.7 3415.22612.2036 3423.45
#Mann= 3 ,-1,0
       0      .1       0  178.86    .045       0  219.79      .1       0
Bank Sta=178.86,219.79
XS Rating Curve= 0 ,0
Exp/Cntr(USF)=0,0
Exp/Cntr=0.3,0.1

Type RM Length L Ch R = 1 ,65416   ,523.1,528.7,532.2
XS GIS Cut Line= 4
 2192304.5105659456381.1789299522192232.35603527456597.642521827
2192188.26159989456790.0546034952192160.20150465456930.355079711
#Sta/Elev= 30
       0 3372.84     8.4 3367.45    28.7 3356.94    37.9 3354.06    46.4 3349.66
    54.8 3347.22    63.2 3343.28    84.3 3328.78    88.5 3327.64   101.5 3326.42
   126.5 3328.79   143.4 3327.19     156 3328.31   189.7 3327.52   202.4 3328.79
   227.7  3328.6   235.9 3326.56   256.4 3327.99   289.3 3327.66  298.363325.224
   324.8  3323.9   343.53325.225   350.8 3329.27     359 3335.45   363.1 3339.08
   371.3 3348.92   375.4 3351.02   453.2 3366.92   538.9 3393.91568.6516 3402.18
#Mann= 4 ,-1,0
       0     .06       0      40      .1       0  298.36    .045       0
   343.5      .1       0
#XS Ineff= 2 , 0
          227.49 3333.07
Permanent Ineff=
       F       F
Bank Sta=298.36,343.5
XS Rating Curve= 0 ,0
Exp/Cntr(USF)=0,0
Exp/Cntr=0.3,0.1

Type RM Length L Ch R = 1 ,64888   ,584.4,572.9,561.7
XS GIS Cut Line= 4
2191845.04654922456161.2278690952191774.91234545456377.474997379
2191719.38943413456523.5879218962191639.56139358456811.588863042
#Sta/Elev= 30
       0 3394.65    35.6 3382.31    50.4 3374.05    71.4 3373.15   105.1  3354.2
   121.9 3341.83   138.7 3326.77   147.1 3323.02   193.4 3321.09   214.4  3322.9
   244.7 3322.49   250.9 3321.59     257 3318.83   265.5 3318.37   295.5 3320.38
   322.3 3319.58   353.2 3319.66   363.9 3322.01   385.2 3322.07   417.4 3318.99
   424.8  3321.5   433.4 3322.44   465.6  3339.1   505.8 3349.51   545.9 3362.77
     554 3363.38   642.3 3394.73   658.4 3398.25   689.5 3410.61   700.6 3416.63
#Mann= 4 ,-1,0
       0     .06       0     160      .1       0   322.3    .045       0
   353.2      .1       0
#XS Ineff= 2 , 0
          216.74 3328.55
Permanent Ineff=
       F       F
Bank Sta=322.3,353.2
XS Rating Curve= 0 ,0
Exp/Cntr(USF)=0,0
Exp/Cntr=0.3,0.1

Type RM Length L Ch R = 1 ,64315   ,379.5,378,359.4
XS GIS Cut Line= 4
2191187.53838889456035.5707540122191187.53838889456319.029827573
2191199.22742286456506.0543709542191225.52774927456731.068274709
#Sta/Elev= 30
       0 3359.61    21.6 3354.25    33.6 3347.35      37 3346.61    61.6 3346.78
    73.6 3343.89   121.6 3337.83   169.6 3321.35   193.6  3317.5   245.6 3318.17
   261.6 3315.55   289.6 3317.52   309.7 3317.34   331.4 3315.09   344.9 3313.71
   365.8 3313.84   372.8 3315.08   405.8 3314.37   421.9 3315.28   433.9 3313.69
   490.1  3316.1   498.2 3322.06   514.4 3340.42   526.3 3349.55   550.2 3359.34
   590.8 3373.55   606.9 3380.35     623    3389   635.1 3392.28697.3943 3426.19
#Mann= 4 ,-1,0
       0     .06       0      90      .1       0   331.4    .045       0
   372.8      .1       0
#XS Ineff= 2 , 0
          241.75 3323.92
Permanent Ineff=
       F       F
Bank Sta=331.4,372.8
XS Rating Curve= 0 ,0
Exp/Cntr(USF)=0,0
Exp/Cntr=0.3,0.1

Type RM Length L Ch R = 1 ,63937   ,417.6,408.5,391.7
BEGIN DESCRIPTION:
new xs added per checkras comments
END DESCRIPTION:
XS GIS Cut Line= 3
2190641.86180813455910.8347659232190933.00066138456519.025354661
2191181.45947333456794.921336019
#Sta/Elev= 30
       0 3355.57    24.8 3352.47    33.5 3352.77   135.6 3343.21   181.4 3340.94
     282 3331.97   326.3 3331.53   361.8 3323.76     450 3321.32     517 3320.59
   521.5 3319.46   530.3 3313.77  536.76 3311.19   570.3 3311.17     589  3312.6
   609.3 3311.02     619 3308.74   660.3 3313.47   708.9 3313.91   779.5 3311.91
   810.5 3314.33     848 3342.03   927.3 3381.33   941.5 3391.15   952.8 3394.21
   962.5 3402.32   978.3 3410.76  1020.8 3437.55  1032.5 3447.91  1045.6 3451.88
#Mann= 5 ,-1,0
       0      .1       0     340     .06       0     450      .1       0
  536.76    .045       0   570.3      .1       0
Bank Sta=536.76,570.3
XS Rating Curve= 0 ,0
Exp/Cntr(USF)=0,0
Exp/Cntr=0.3,0.1

Type RM Length L Ch R = 1 ,63528   ,319.4,317.2,315.5
XS GIS Cut Line= 4
2190012.79047578456444.686942657 2190340.0834267456511.898887934
2190804.72252666456839.1918388512191053.11449834457034.983157703
#Sta/Elev= 30
       0 3386.64   108.3 3365.73   186.2 3346.89   219.9 3342.42   232.1 3337.74
   264.8 3335.96   293.4 3325.97     326 3332.43   363.6 3327.65   383.2 3329.65
   537.8 3324.26     574  3315.8   603.3 3316.87   622.9 3312.02   671.8 3312.61
   681.6 3309.44   705.4  3309.2  715.713306.256   739.9 3305.28  765.263306.254
   774.6 3309.56   828.9 3309.05   851.8  3306.3  1023.1 3310.44  1054.3 3328.84
  1091.5 3355.44  1117.1 3377.68  1131.3 3386.17  1162.7 3401.271218.742 3423.05
#Mann= 5 ,-1,0
       0      .1       0     200     .06       0     330      .1       0
  715.71    .045       0  765.26      .1       0
#XS Ineff= 2 , 0
                          875.01         3311.39
Permanent Ineff=
       F       F
Bank Sta=715.71,765.26
XS Rating Curve= 0 ,0
Exp/Cntr(USF)=0,0
Exp/Cntr=0.3,0.1

Type RM Length L Ch R = 1 ,63211   ,365.8,368.3,367.3
XS GIS Cut Line= 4
2190185.20372671456874.2589407352190407.29537198456953.159919974
2190638.15379271457096.350585999 2190883.6235059457219.085442593
#Sta/Elev= 30
       0 3440.97    41.4 3419.67    54.7 3410.05    70.4 3401.46   100.8 3380.05
   117.8 3362.77   130.5 3352.48   134.7 3350.35   147.5 3350.77     156 3348.87
   185.7 3321.63   211.3 3304.36   236.7 3304.95   269.7 3302.99   297.9 3306.76
   323.5 3306.37   340.3 3305.47  345.833301.865   363.8 3300.29  393.223301.865
   410.6 3305.71   503.6 3303.43     523 3304.57   553.9 3303.27   563.3 3305.31
   604.9 3304.67   612.5 3307.03   639.3 3326.55   666.1 3335.98781.7941 3350.76
#Mann= 5 ,-1,0
       0      .1       0     130     .06       0  235.69      .1       0
  345.83    .045       0  393.22      .1       0
#XS Ineff= 2 , 0
          299.56 3311.88  564.76         3310.91
Permanent Ineff=
       F       F
Bank Sta=345.83,393.22
XS Rating Curve= 0 ,0
Exp/Cntr(USF)=0,0
Exp/Cntr=0.3,0.1

Type RM Length L Ch R = 1 ,62843   ,460.3,466,469.8
XS GIS Cut Line= 4
2190193.97050218457233.6967350452190313.78310029457318.442231264
2190588.47539838457508.3890331352190708.28799648457607.745821806
#Sta/Elev= 30
       0 3347.24    17.4 3338.82      37 3338.42    51.7 3330.43    90.2 3318.23
   105.6 3311.19   121.7 3302.13   130.1 3299.47     174 3299.56  195.833297.182
   227.5 3296.42   233.8 3297.39   242.1 3300.65     250 3301.16   261.5 3299.14
   285.8 3298.34   295.6 3296.41   320.1 3296.13   349.1 3297.77   358.8 3300.63
   371.8 3302.41   397.7  3310.1   411.8 3312.36   436.6 3320.69   452.3  3327.8
   465.8 3329.85   506.6 3344.19   588.5 3376.51   620.6 3391.88636.3737 3395.89
#Mann= 5 ,-1,0
       0      .1       0      20     .06       0     140      .1       0
  195.83    .045       0   233.8      .1       0
Bank Sta=195.83,233.8
XS Rating Curve= 0 ,0
Exp/Cntr(USF)=0,0
Exp/Cntr=0.3,0.1

Type RM Length L Ch R = 1 ,62377   ,494.9,488.4,479.8
XS GIS Cut Line= 4
2189890.05561919457517.1558086062190082.92467955457698.335835006
2190205.65953615 457823.992950092190293.32729086457917.505221781
#Sta/Elev= 30
       0 3349.59      10 3346.54    29.2 3337.19    49.6 3329.49    63.8 3326.01
    79.7 3319.89    99.4 3319.78   116.9 3315.48   123.2 3311.55  148.793290.638
   169.5 3289.37   182.6 3290.44   198.7 3292.76   227.9 3291.53   239.6 3294.08
   261.9 3295.73   295.8    3295   326.9 3289.12     386 3291.95   397.2 3290.78
   402.8 3291.44   425.2  3309.3   440.1 3318.94   447.4 3325.04   469.3 3337.51
   480.3 3341.61   496.7  3351.1     508 3355.34   541.9 3372.27568.4539 3379.21
#Mann= 4 ,-1,0
       0      .1       0      30     .06       0  148.79    .045       0
   182.6      .1       0
Bank Sta=148.79,182.6
XS Rating Curve= 0 ,0
Exp/Cntr(USF)=0,0
Exp/Cntr=0.3,0.1

Type RM Length L Ch R = 1 ,61888   ,360.1,357.7,354.1
XS GIS Cut Line= 4
 2189430.9559854 457854.518184392189691.34204185   458002.250718
2189913.43368711458107.4520236522190053.70209465458165.897193458
#Sta/Elev= 30
       0 3334.55   38.06 3324.82   51.99 3323.08   65.79 3319.37   90.87    3312
  102.61 3305.78  123.15 3305.01  134.89 3302.37  153.17 3302.35  175.62  3298.8
  235.95 3295.74  249.74 3292.02  317.22 3289.07  322.43 3287.67  329.23 3283.87
  335.71  3282.9  353.26 3283.64  397.67 3286.29  431.35 3284.98  446.36 3282.22
  464.06 3284.48  512.75 3285.64  570.41 3291.98  576.07 3294.83  600.09 3313.55
  626.09 3336.83  630.43 3339.18  647.76  3343.5  667.83 3352.98  697.08 3362.73
#Mann= 5 ,-1,0
       0      .1       0     100     .06       0     220      .1       0
  329.23    .045       0  353.26      .1       0
Bank Sta=329.23,353.26
XS Rating Curve= 0 ,0
Exp/Cntr(USF)=0,0
Exp/Cntr=0.3,0.1

Type RM Length L Ch R = 1 ,61531   ,444.6,431.8,415
XS GIS Cut Line= 4
2189369.89360791458247.7204311872189697.18655883458320.776893446
2189907.58917013458341.2327028782190001.10144182458352.921736839
#Sta/Elev= 30
       0    3332    10.5 3328.48    46.7 3321.49    80.2 3310.81    88.4 3306.38
   100.7 3297.26     113 3291.13   121.2 3291.69   145.8 3290.24   158.1 3287.17
   174.5 3284.94   227.6 3283.38     240 3281.93   305.6 3283.56     322 3282.33
   338.5 3283.62   346.4 3283.26   366.5 3279.05   382.6 3280.15   431.7 3279.76
   454.9 3278.32   471.8 3278.54  478.753279.926     485 3283.41   511.2 3305.19
   515.2 3307.02   539.9 3313.82   571.5 3319.68   579.5 3322.15640.9821 3347.43
#Mann= 5 ,-1,0
       0      .1       0     160     .06       0     260      .1       0
   431.7    .045       0  478.75      .1       0
#XS Ineff= 2 , 0
          339.98  3287.7
Permanent Ineff=
       F       F
Bank Sta=431.7,478.75
XS Rating Curve= 0 ,0
Exp/Cntr(USF)=0,0
Exp/Cntr=0.3,0.1

Type RM Length L Ch R = 1 ,61099   ,637.3,645.4,651.9
XS GIS Cut Line= 4
2189577.37396073458817.5608368012189694.26430034458770.804700956
 2189916.3559456 458630.536293422190044.93531918 458539.94628022
#Sta/Elev= 30
       0 3304.79    30.1 3299.46    54.7 3296.41    76.3 3296.53    97.8 3294.35
   119.3 3293.94   128.5 3292.61   137.2 3289.55   151.8 3276.64   156.5 3274.69
   174.9 3275.13   194.4 3273.27   212.5 3273.62   222.8 3272.42   238.6 3273.28
   287.9  3273.1   303.2 3275.24   312.7 3274.02   326.9 3276.59   346.2 3277.08
   369.1 3275.44   374.2 3276.61   400.9 3286.05   422.6 3304.25   432.5 3310.77
   442.2  3314.6   466.6 3327.38     487 3333.93   532.9 3355.39545.8601 3360.29
#Mann= 5 ,-1,0
       0      .1       0     120     .06       0  155.89      .1       0
   212.5    .045       0   238.6      .1       0
#XS Ineff= 2 , 0
                          346.26         3280.91
Permanent Ineff=
       F       F
Bank Sta=212.5,238.6
XS Rating Curve= 0 ,0
Exp/Cntr(USF)=0,0
Exp/Cntr=0.3,0.1

Type RM Length L Ch R = 1 ,60453   ,526.5,529.6,533
XS GIS Cut Line= 4
2189594.90751167459413.7015688272189869.59980976459326.033814117
2190170.59243426459241.2883178982190328.39439274459191.609923562
#Sta/Elev= 30
       0 3291.22    55.5 3287.19    67.5 3280.85    81.1 3278.65    93.7 3273.63
   144.1 3272.38   198.8 3273.93     221 3269.48   244.9  3267.6   311.8 3270.51
   324.3 3269.79   340.9 3264.64   352.7 3267.46   361.7 3267.98   390.8 3267.81
   411.1 3265.85     424 3267.78   448.9 3267.86     463 3265.81   473.9 3264.85
   511.3 3265.84   536.2 3265.23   552.8 3269.98   568.5 3278.07   589.4 3292.65
   611.1 3305.25   711.7 3334.18   732.7 3341.79   753.7 3346.86 766.475 3351.57
#Mann= 5 ,-1,0
       0      .1       0     130     .06       0     230      .1       0
     463    .045       0   511.3      .1       0
#XS Ineff= 2 , 0
           316.3 3273.18
Permanent Ineff=
       F       F
Bank Sta=463,511.3
XS Rating Curve= 0 ,0
Exp/Cntr(USF)=0,0
Exp/Cntr=0.3,0.1

Type RM Length L Ch R = 1 ,59924   ,512,507.5,495.3
XS GIS Cut Line= 4
2189667.96397393459846.195825395  2189948.500789459822.817757472
2190269.94922293459770.2171046472190439.44021537459723.460968801
#Sta/Elev= 30
       0 3296.57    27.1 3292.14    40.4 3287.72    60.4 3288.41    68.4 3285.99
   108.6 3280.84   148.7 3270.24   184.8 3264.98   249.1 3262.18   271.6 3264.45
   289.3    3264     314 3258.06     342  3260.1   362.2 3257.52   370.3 3259.67
   390.6 3261.25   459.5 3259.28   471.7 3260.33     496 3258.26   516.6 3258.31
   544.6 3258.65   556.8 3263.56   599.6 3265.27   609.9 3267.57   630.3 3280.22
   684.2 3320.44   709.1 3330.56   729.9 3343.51   767.2 3372.26783.0548 3386.13
#Mann= 5 ,-1,0
       0      .1       0      50     .06       0     150      .1       0
     496    .045       0   516.6      .1       0
#XS Ineff= 2 , 0
          278.41 3270.06
Permanent Ineff=
       F       F
Bank Sta=496,516.6
XS Rating Curve= 0 ,0
Exp/Cntr(USF)=0,0
Exp/Cntr=0.3,0.1

Type RM Length L Ch R = 1 ,59416   ,461.4,466.4,473.6
XS GIS Cut Line= 4
2189811.15463995460261.1565310212189960.18982296460223.167170647
2190202.73727766 460158.877483862190363.46149462460144.266191408
#Sta/Elev= 30
       0 3304.25    69.9 3296.62    87.7 3295.91   104.3 3293.57   120.8 3288.32
   132.4 3289.16   157.9 3288.69   182.8 3284.85   186.9 3283.67     191 3281.11
   203.4 3269.32   211.7  3262.7   215.9 3260.03   224.1 3256.59   240.7 3253.98
   257.2 3254.57  274.343252.586   315.7 3250.97   327.6 3251.07  338.533252.586
   360.7 3257.63   381.4 3256.95   410.2 3258.71   414.2 3260.58   422.2 3268.77
   430.3 3274.92   458.4 3291.26   503.3 3307.29   534.7 3315.64566.1109 3329.51
#Mann= 6 ,-1,0
       0     .12       0      10      .1       0      50     .06       0
   213.8      .1       0  274.34    .045       0  338.53      .1       0
Bank Sta=274.34,338.53
XS Rating Curve= 0 ,0
Exp/Cntr(USF)=0,0
Exp/Cntr=0.3,0.1

Type RM Length L Ch R = 1 ,58950   ,550,518.5,494.4
XS GIS Cut Line= 4
2189875.44432674 460664.486831072190009.86821729460629.361100802
2190193.97050218460629.3611008022190360.53923613460582.604964957
#Sta/Elev= 30
       0 3331.48   16.42 3322.39   22.98 3317.96   33.83 3313.07   75.17 3291.18
   95.09 3286.43  112.38 3283.99  133.05 3277.59  141.43  3278.3  157.24 3276.94
  177.24 3270.18  181.24  3267.9  185.24 3264.67  201.24  3249.7  207.07 3247.15
  213.24 3246.07  253.24 3245.39  265.06 3247.04  281.24 3250.05  305.24    3253
  321.24 3252.69   346.1 3250.57  357.42 3251.05  412.58 3272.25  416.73 3272.96
  428.78 3273.12     445 3277.64  449.97 3277.72  487.36 3286.32  496.05  3287.2
#Mann= 4 ,-1,0
       0      .1       0      90     .07       0  207.07    .045       0
  265.06      .1       0
#XS Ineff= 2 , 0
                          307.82         3255.15
Permanent Ineff=
       F       F
Bank Sta=207.07,265.06
XS Rating Curve= 0 ,0
Exp/Cntr(USF)=0,0
Exp/Cntr=0.3,0.1

Type RM Length L Ch R = 1 ,58431   ,424.1,436.8,450.2
XS GIS Cut Line= 4
2190042.01306069461205.0460233962190357.61697764461076.466649822
 2190521.2634531460930.3537253062190620.62024177460807.618868712
#Sta/Elev= 30
       0 3296.37    41.2 3287.79   126.9 3273.06   170.8 3270.13   196.7 3266.12
   218.3 3264.34   256.3 3262.51   285.9 3258.99   300.4 3253.21   328.3 3253.96
   338.9 3252.87   351.7  3249.6   390.3 3246.21   413.9 3245.46  433.843241.348
   440.7 3240.18   462.2 3239.98   489.4 3240.04  497.713241.348   515.8 3242.95
   531.9 3253.19   555.9  3270.8   571.6  3280.6   577.1 3282.98   590.2 3285.16
   597.7 3288.26   639.9 3299.52   660.2 3306.55   672.9 3308.75718.0847 3324.75
#Mann= 5 ,-1,0
       0      .1       0     190     .06       0  410.79      .1       0
  433.84    .045       0  497.71      .1       0
Bank Sta=433.84,497.71
XS Rating Curve= 0 ,0
Exp/Cntr(USF)=0,0
Exp/Cntr=0.3,0.1

Type RM Length L Ch R = 1 ,57995   ,275.2,272.7,275.7
XS GIS Cut Line= 4
 2190220.2708286461529.4167158222190456.97376631461432.982185641
2190714.13251346461336.5476554612190860.24543798461251.802159241
#Sta/Elev= 30
       0 3273.93    43.1 3264.25      69 3263.13    90.6 3259.38   104.5 3252.45
   112.2 3250.22   122.9 3250.37   142.4 3253.45   189.9 3254.13   228.8 3251.74
   292.1 3250.94   297.5 3248.67     306 3241.25   323.1 3242.19   344.5 3238.71
   395.7 3239.58     435 3236.19   451.3 3237.25   472.3 3236.76   481.2 3235.85
  494.853237.271   506.8 3250.79   519.6  3262.1   534.2 3273.56   544.9 3279.67
   584.8 3290.91   603.7 3293.85   648.2 3306.06   657.1 3310.71699.1495 3327.14
#Mann= 7 ,-1,0
       0      .1       0     100     .12       0     200      .1       0
  305.59     .06       0  415.59      .1       0   472.3    .045       0
  494.85      .1       0
#XS Ineff= 2 , 0
          318.39    3246
Permanent Ineff=
       F       F
Bank Sta=472.3,494.85
XS Rating Curve= 0 ,0
Exp/Cntr(USF)=0,0
Exp/Cntr=0.3,0.1

Type RM Length L Ch R = 1 ,57722   ,235.1,231.5,232
BEGIN DESCRIPTION:
new xs added per checkras comments
END DESCRIPTION:
XS GIS Cut Line= 2
2190318.91709316461740.4355565842190968.97222957461473.746269853
#Sta/Elev= 30
       0 3283.55    74.9 3263.93    86.2 3259.31   113.8 3252.18   152.7 3245.64
     170 3244.06   221.9 3242.97   234.8 3238.03   243.5 3236.79   285.5 3238.76
   300.8 3235.62   338.6 3235.09   362.9 3232.33   373.2 3231.84   381.8 3232.27
   403.4 3232.87   420.4 3235.81   433.7 3236.44   463.3 3234.91   472.6 3232.87
   489.9 3233.38   494.9 3235.25   507.2  3243.7   520.2 3249.88   533.2    3258
   550.4 3273.59   563.4 3281.39   598.7 3292.59   670.8 3312.01   702.6 3322.78
#Mann= 5 ,-1,0
       0     .12       0     200     .06       0     310      .1       0
   362.9    .045       0   381.8      .1       0
#XS Ineff= 2 , 0
          277.63 3248.34
Permanent Ineff=
       F       F
Bank Sta=362.9,381.8
XS Rating Curve= 0 ,0
Exp/Cntr(USF)=0,0
Exp/Cntr=0.3,0.1

Type RM Length L Ch R = 1 ,57490   ,545.3,566.1,597.6
XS GIS Cut Line= 4
 2190372.2282701461900.5435440932190725.82154742461830.409340326
2190877.77898892461739.8193271262191094.02611721461561.561559216
#Sta/Elev= 30
       0 3281.73    48.9 3264.27    97.8 3250.73   167.1 3242.76   187.5  3242.4
   216.1 3233.32   232.4 3233.22   269.1 3237.53   277.2 3235.89   309.9 3236.93
   338.4 3234.45   358.8 3235.34   377.2 3233.64   403.9 3233.45  413.43  3230.6
   428.4 3229.22   456.4 3229.34  463.273230.603   479.6 3234.68   506.1 3235.84
   541.5    3244     573 3245.89   579.3 3247.31     595 3252.84     617 3264.18
   646.1 3285.68     661 3294.55   680.5 3299.98   794.5 3321.02817.6404 3328.05
#Mann= 4 ,-1,0
       0      .1       0     340     .06       0  413.43    .045       0
  463.27      .1       0
#XS Ineff= 2 , 0
          357.93 3239.82
Permanent Ineff=
       F       F
Bank Sta=413.43,463.27
XS Rating Curve= 0 ,0
Exp/Cntr(USF)=0,0
Exp/Cntr=0.3,0.1

Type RM Length L Ch R = 1 ,56924   ,572,560.5,550
XS GIS Cut Line= 4
2190369.30601161462309.6597327392190670.29863611462300.892957268
2190895.31253986462368.1049025452191123.24870211 462318.42650821
#Sta/Elev= 30
       0 3297.73    50.9 3276.78    93.1 3261.94   110.9 3258.49   146.9 3241.83
   163.2 3236.05   178.2 3232.43     203 3234.18     239 3226.54     271  3229.2
   307.3 3229.54   336.5  3225.7  365.083224.489   373.6 3223.37   389.6 3224.43
   453.4 3225.03   474.2  3222.9   486.8 3223.37   503.5 3226.33   507.6 3227.96
   527.9 3241.02     545 3257.59   553.2  3262.7   557.3 3263.95   577.8 3266.69
   619.8 3267.71     631 3269.31   643.3 3269.31   704.7 3274.18769.2449 3281.87
#Mann= 7 ,-1,0
       0      .1       0     240     .06       0  331.12      .1       0
  361.12     .06       0  365.08    .045       0   389.6     .06       0
  441.12      .1       0
#XS Ineff= 2 , 0
          303.08 3232.85
Permanent Ineff=
       F       F
Bank Sta=365.08,389.6
XS Rating Curve= 0 ,0
Exp/Cntr(USF)=0,0
Exp/Cntr=0.3,0.1

Type RM Length L Ch R = 1 ,56364   ,337.2,313.9,274.1
XS GIS Cut Line= 4
2190515.41893612462891.1891723132190816.41156062462797.676900623
2191012.20287948462733.3872138362191193.38290588462458.694915745
#Sta/Elev= 30
       0 3306.25    67.8  3280.4    88.8  3275.1   134.8 3258.85   143.2    3254
   158.8  3241.3   168.6 3235.79     182 3225.55   190.8 3220.89   197.7 3220.27
   214.4 3223.01   264.7 3222.67   281.4 3220.92   331.8 3222.67   352.8  3221.6
   369.7 3218.46   385.1 3219.38  393.253218.048   407.3  3216.6  437.473218.047
   445.4  3224.1   449.7 3225.78   524.3 3231.49   558.9 3242.01   593.4 3248.71
   674.8  3257.1   698.8 3255.19   751.5 3263.55   840.9 3273.43850.3229 3273.33
#Mann= 5 ,-1,0
       0      .1       0     200     .06       0     300      .1       0
  393.25    .045       0  437.47      .1       0
#XS Ineff= 2 , 0
          320.48 3227.27
Permanent Ineff=
       F       F
Bank Sta=393.25,437.47
XS Rating Curve= 0 ,0
Exp/Cntr(USF)=0,0
Exp/Cntr=0.3,0.1

Type RM Length L Ch R = 1 ,56050   ,339.5,331.8,316.4
XS GIS Cut Line= 4
 2190965.6622579463252.4507673852191044.34772287463069.446940223
2191102.79289268462818.132710055 2191216.7609738462476.228466687
#Sta/Elev= 30
       0 3280.84   77.58 3267.65      95  3263.5  112.41 3262.43  138.54 3256.88
  160.31 3244.35  164.66 3243.33  169.02 3244.79  177.72 3231.95  195.14 3221.83
   215.9  3221.5  225.94 3215.01  236.44 3212.75  265.92 3214.81  277.51 3217.34
  304.39 3217.34  330.89  3216.2  343.21 3213.19  363.75 3218.34  392.53 3218.85
  413.03 3226.31  425.35 3228.22   454.1 3226.58  479.31 3227.22  529.91 3244.35
  629.83 3254.35  673.26 3260.51  685.91 3260.18  787.11 3272.44  817.62 3274.49
#Mann= 5 ,-1,0
       0      .1       0     170     .06       0  225.94    .045       0
  265.92     .06       0   369.2      .1       0
Bank Sta=225.94,265.92
XS Rating Curve= 0 ,0
Exp/Cntr(USF)=0,0
Exp/Cntr=0.3,0.1

Type RM Length L Ch R = 1 ,55718   ,288.7,325.3,362.8
BEGIN DESCRIPTION:
new xs added per checkras comment
END DESCRIPTION:
XS GIS Cut Line= 3
2191288.30886721463280.5455427072191379.03656255463020.513487296
2191336.91298971462734.559233215
#Sta/Elev= 30
       0 3243.87    45.9 3238.79    79.8 3237.22     101 3232.99     118 3231.16
   143.4 3224.73   160.3 3223.02     173 3218.07   184.7 3215.42   194.2 3211.71
     213 3212.52   232.3 3209.73   253.5 3212.05   266.4 3209.52   278.8 3211.81
   290.9 3212.16   323.2 3210.72   331.3 3208.39   339.4 3207.89     369 3208.41
   386.6 3210.29   400.1 3210.53   416.2 3217.39   432.4 3221.01   440.5 3223.95
   467.6 3229.04   488.8 3231.85   509.2 3238.16   545.6 3242.28   564.4 3243.41
#Mann= 5 ,-1,0
       0      .1       0      90     .06       0  295.41      .1       0
   331.3    .045       0     369      .1       0
#XS Ineff= 2 , 0
          210.25  3215.1
Permanent Ineff=
       F       F
Bank Sta=331.3,369
XS Rating Curve= 0 ,0
Exp/Cntr(USF)=0,0
Exp/Cntr=0.3,0.1

Type RM Length L Ch R = 1 ,55393   ,497.8,504,500
XS GIS Cut Line= 4
 2191286.2804584463294.0103219142191531.99212227463174.210605201
 2191650.5693929463113.0883007562191811.93227663463034.851751066
#Sta/Elev= 30
       0 3244.89    37.9  3236.3    58.9 3233.75      84 3228.36    97.8 3227.53
   120.6 3219.71   148.6 3214.88   184.6 3213.56   208.5 3208.01   246.9 3209.74
   260.2 3208.47   300.6 3208.05  315.933204.876   345.5 3203.59  363.893204.876
   377.1 3206.94   380.4 3208.75   404.1 3226.12   421.9 3243.85   426.3 3246.35
   439.7 3250.74   448.6 3251.34   488.6 3264.05   497.7  3262.7   501.9 3263.29
   519.7 3271.42   544.1 3274.94   555.2 3282.03   562.4  3284.9586.0936 3289.59
#Mann= 5 ,-1,0
       0      .1       0     120     .06       0     230      .1       0
  315.93    .045       0  363.89      .1       0
#XS Ineff= 2 , 0
          243.83 3213.64
Permanent Ineff=
       F       F
Bank Sta=315.93,363.89
XS Rating Curve= 0 ,0
Exp/Cntr(USF)=0,0
Exp/Cntr=0.3,0.1

Type RM Length L Ch R = 1 ,54889   ,555,556.5,554.5
XS GIS Cut Line= 4
2191342.41808888463753.2554269592191593.73231905463653.898638288
2191795.36815488463566.2308835782192005.77076619463458.107319436
#Sta/Elev= 30
       0 3246.83     6.2  3243.2    27.7 3234.58    44.9 3228.39    53.5 3227.16
    70.7 3226.93    87.2 3224.63   167.9 3219.29   225.6 3217.48     260 3218.43
   290.4  3218.6   299.1 3213.49   309.1 3203.62   315.2 3199.45   341.93193.449
   364.5 3192.45  395.653193.448   421.2 3196.27     443 3196.89   461.1 3202.88
   504.5 3204.07   530.1 3214.87   562.4  3237.3   577.6 3246.52   594.5 3254.83
   603.4 3258.04   625.9 3261.93   651.9 3264.02   679.9 3269.31  726.67 3275.48
#Mann= 5 ,-1,0
       0      .1       0     260     .06       0   341.9    .045       0
  395.65     .06       0  420.24      .1       0
Bank Sta=341.9,395.65
XS Rating Curve= 0 ,0
Exp/Cntr(USF)=0,0
Exp/Cntr=0.3,0.1

Type RM Length L Ch R = 1 ,54332   ,450.3,447,445.6
XS GIS Cut Line= 4
2191614.18812848464220.8167854112191710.62265866464191.594200508
 2191970.7036643464092.2374118372192306.76339069463881.834800534
#Sta/Elev= 30
       0 3254.74    18.8 3241.47    39.7  3234.6    60.6 3232.66      94 3209.98
   115.3  3201.2   132.4 3198.93   145.2 3190.34   159.6 3190.67   175.2 3188.31
   192.3 3190.36   209.2 3188.83   230.9 3189.94     278 3188.65  285.033186.812
   311.4 3185.07  329.333186.813   350.8 3197.69   357.9 3198.61   388.3 3198.75
   405.7 3196.03   434.7 3195.94   472.4 3204.39   576.9 3206.82   593.3 3204.57
     635 3205.27   659.4 3212.67   682.9 3216.51   706.5 3223.86775.6695  3239.1
#Mann= 7 ,-1,0
       0      .1       0  180.76     .06       0  285.03    .045       0
  329.33      .1       0  389.18     .12       0  629.18      .1       0
  739.18     .06       0
#XS Ineff= 2 , 0
          194.71 3194.06
Permanent Ineff=
       F       F
Bank Sta=285.03,329.33
XS Rating Curve= 0 ,0
Exp/Cntr(USF)=0,0
Exp/Cntr=0.3,0.1

Type RM Length L Ch R = 1 ,53885   ,455,437,415.7
XS GIS Cut Line= 4
2191722.31169262464615.3216816052191824.59073979464583.176838211
2192040.83786807464489.6645665212192473.33212464464323.095832573
#Sta/Elev= 30
       0 3268.08    39.7 3258.98    64.8 3241.03    85.8  3224.2   102.6 3212.87
   112.2 3202.19   132.4 3185.92   159.1 3185.19  167.193181.127   193.6 3179.85
  210.713181.126   233.1 3185.22   241.9 3184.52   266.6 3186.01   284.9 3189.48
   337.7 3190.51   379.8 3189.69   457.8 3192.16   555.6 3196.81   571.7 3200.16
   620.7 3200.45   645.9  3202.6   676.4    3200   693.6 3200.12   698.6 3201.04
     715 3210.87   736.5 3219.28   766.5 3220.56   783.6 3224.27806.2728  3226.5
#Mann= 6 ,-1,0
       0     .12       0      70     .06       0  167.19    .045       0
  210.71      .1       0  702.81     .06       0  802.81      .1       0
Bank Sta=167.19,210.71
XS Rating Curve= 0 ,0
Exp/Cntr(USF)=0,0
Exp/Cntr=0.3,0.1

Type RM Length L Ch R = 1 ,53448   ,251.2,234.2,215.7
BEGIN DESCRIPTION:
structure xs 4
END DESCRIPTION:
XS GIS Cut Line= 4
2192033.64305744465036.0758657982192110.51695217464949.418020829
2192213.94728326464788.6816954832192499.07954736464360.983299345
#Sta/Elev= 30
       0  3226.4    57.3 3220.45      68 3214.72    77.5 3206.63   116.1 3180.97
   120.9 3179.84   143.3 3179.82  150.073176.774   155.9  3175.2   187.5 3174.81
  197.943176.775   201.7 3179.01   207.6 3179.61   281.5 3181.18   296.9 3185.45
   330.4 3188.09   417.8 3191.56   431.4 3190.39   475.5 3194.22   537.1 3194.96
   609.2 3201.71   628.3 3204.59   642.8 3208.67   664.3 3211.21     691 3212.09
   719.8 3210.29   724.6 3211.46     739 3220.45   749.5 3224.93821.0093 3230.19
#Mann= 7 ,-1,0
       0      .1       0      70     .06       0  150.07    .045       0
  197.94     .06       0  235.84      .1       0  566.98     .06       0
  776.98      .1       0
#XS Ineff= 2 , 0
                          259.91         3184.53
Permanent Ineff=
       F       F
Bank Sta=150.07,197.94
XS Rating Curve= 0 ,0
Exp/Cntr(USF)=0,0
Exp/Cntr=0.5,0.3

Type RM Length L Ch R = 1 ,53214   ,71.3,66.5,63.3
BEGIN DESCRIPTION:
structure xs 3
END DESCRIPTION:
XS GIS Cut Line= 5
2192192.98167561465235.9479920982192355.11570813465078.007081106
2192360.70653684464871.1464189212192388.66068038464549.673768229
2192506.06808324464367.971835229
#Sta/Elev= 30
       0 3194.22    21.2 3193.22      38 3186.66    54.7 3184.09      67 3179.27
    77.8 3177.45   164.5 3177.27   179.6 3175.61   263.2 3177.15   279.2    3179
  294.993174.482   327.2 3173.17   338.33174.481   359.2 3182.35   451.3 3184.89
   515.6 3189.65   587.8 3190.95   620.7 3196.81   699.9 3197.79   736.4 3201.95
     756 3202.14   779.1 3207.64   802.3 3210.03   842.3 3210.53   857.2 3206.78
   870.9 3206.31   885.1 3208.82   895.1 3215.03     909 3220.59972.3018 3230.62
#Mann= 5 ,-1,0
       0     .06       0  294.99    .045       0   338.3      .1       0
  563.28     .06       0  905.97      .1       0
#XS Ineff= 3 ,-1
   15.42  160.79 3180.92   168.5  274.23 3174.45     358972.3018 3174.53
Permanent Ineff=
       F       F       F
Bank Sta=294.99,338.3
XS Rating Curve= 0 ,0
Exp/Cntr(USF)=0,0
Exp/Cntr=0.5,0.3
